--- ROARCK.prj (project) ---

Proj Title=ROARCK
Current Plan=p01
Default Exp/Contr=0,0
English Units
Geom File=g01
Flow File=f01
Plan File=p01
BEGIN DESCRIPTION:
----------MODEL BY WOOD PLC 2022----------
AFH study
Randolph County, WV
HEC-RAS Version: RAS 6.2
Vertical Datum: NAVD88
Projection: NAD 1983 StatePlane West Virginia S FIPS 4702 (US Feet)
Terrain: 1-meter LIDAR (FEMA Region III 3DEP collected 2016-2018)
Land Use: 2019 NLCD
Hydrologic Method:
WV SIR2010-5033 regression equations
Additional Model Notes:
None
END DESCRIPTION:
DSS Export Rating Curves= 0
DSS Export Rating Curve Sorted= 0
DSS Export Volume Flow Curves= 0
DXF OffsetX= 0
DXF OffsetY= 0
DXF ScaleX= 0
DXF ScaleY= 0

--- ROARCK.p01 (plan) ---

Plan Title=Floodplain
Program Version=4.00
Geom File=g01
Flow File=f01
K Sum by GR=0
Std Step Tol=0.01
Critical Tol=0.01
Num of Std Step Trials=20
Max Error Tol=0.3
Flow Tol Ratio=0.001
Split Flow NTrial=30
Split Flow Tol=0.02
Split Flow Ratio=0.02
Log Output Level=0
Friction Slope Method=1
Unsteady Friction Slope Method=2
Unsteady Bridges Friction Slope Method=1
Global Log Level=0
CheckData=False
Run HTab=0
Run UNet=0
Run PostProcess=0
UNET Theta=0
UNET Theta Warmup=0
UNET ZTol=0
UNET ZSATol=0
UNET MxIter=0
UNET MaxInSteps=0
UNET DtIC=0
UNET DtMin=0
UNET MaxCRTS=0
UNET WFStab=0
UNET SFStab=0
UNET WFX=0
UNET SFX=0
UNET DSS MLevel=0
UNET DZMax Abort=0
UNET Convert EG Bridges=0
UNET Use Existing IB Tables=0
UNET Froude Limit=0
UNET Froude Power=0
Write IC File=0
Echo Input=False
Echo Output=False
Write Detailed=0

--- ROARCK.f01 (steady flow) ---

Flow Title=Flow
Program Version=6.20
Number of Profiles= 1
Profile Names=P100yr
River Rch & RM=ROARCK,Main,75812
     550
River Rch & RM=ROARCK,Main,69434
     622
River Rch & RM=ROARCK,Main,64036
     694
River Rch & RM=ROARCK,Main,60979
     873
River Rch & RM=ROARCK,Main,57717
    1280
River Rch & RM=ROARCK,Main,56825
    1430
River Rch & RM=ROARCK,Main,51265
    2300
River Rch & RM=ROARCK,Main,46906
    2560
River Rch & RM=ROARCK,Main,33666
    3040
River Rch & RM=ROARCK,Main,29243
    3460
River Rch & RM=ROARCK,Main,22240
    3850
River Rch & RM=ROARCK,Main,10606
    4370
Boundary for River Rch & Prof#=ROARCK,Main            , 1
Up Type= 0
Dn Type= 3
Dn Slope=0.01168
DSS Import GetInterval= 0
DSS Import GetPeak= 0
DSS Import FillOption= 0

--- ROARCK.g01 (geometry) ---

Geom Title=Geometry
Program Version=6.20

River Reach=ROARCK          ,Main
Reach XY= 30
     2263533.921      673806.236     2261311.067      673965.128
2258815.18633084 676487.16165418     2256614.299      675417.174
     2255626.037      675941.542     2253972.106      678116.975
     2255042.144      680338.392     2253515.996      684957.786
     2254503.312      685613.405     2257191.924      683899.492
     2259504.747      683802.879     2259624.628        684762.6
     2258512.784      685320.055 2260332.4636888685316.998957349
     2260813.803      686922.577     2262666.209      687690.272
2262471.66992582688390.797820863     2265329.944      688579.396
     2265464.752      692363.204     2262013.973      692870.613
     2262644.314      693926.152     2263877.497      693901.263
     2263087.556      694778.107     2264376.064      694910.825
     2266137.552      697978.784     2267794.181      698927.097
     2266801.773       701160.75     2268164.994      703939.873
     2266502.607      705957.919     2267072.221       706909.63

Type RM Length L Ch R = 1 ,75812   ,278.5,275.5,262.8
XS GIS Cut Line= 4
 2263742.1144084673409.888912911 2263545.9263123673780.770687697
2263525.35582057673822.2384301152263561.55121703674208.481086248
#Sta/Elev= 30
       0 2646.28    24.6 2643.82    44.4 2639.19   132.5 2632.84   171.2 2631.61
   189.3 2633.89   196.2 2633.79     288 2629.99   338.6 2626.46   352.2  2623.7
   361.2 2618.93   365.7 2617.66   415.5 2615.45  438.642612.206     457 2611.03
  462.532612.205   468.8 2613.75   488.9 2613.99     513 2616.55     517 2617.77
   529.9 2625.87   553.2 2633.69   597.4 2644.62   649.6 2665.64   673.2 2673.64
   693.8 2679.75   749.7 2692.57   778.2 2700.98   798.3 2708.14   853.8 2724.17
#Mann= 3 ,-1,0
       0      .1       0  438.64    .045       0  462.53      .1       0
Bank Sta=438.64,462.53
XS Rating Curve= 0 ,0
Exp/Cntr=0.3,0.1

Type RM Length L Ch R = 1 ,75537   ,234.6,234.1,232.9
XS GIS Cut Line= 4
2263374.71119545673423.7003309942263287.61236322673749.570099843
2263310.13792328673887.5952572132263394.81061423674189.470010492
#Sta/Elev= 30
       0 2637.85    30.5  2633.7    38.8 2630.79    51.2 2630.87    76.1 2626.11
     134 2622.28   142.3 2622.63   156.8 2619.99   226.7 2618.16     245 2616.57
   286.7 2615.29   320.2 2609.82     345 2604.19   389.6 2605.36   409.9 2604.86
  419.592601.555   430.1 2599.59   440.1 2601.54   458.5 2604.37   474.7 2604.48
   486.6 2609.09   503.7 2617.98   558.8 2634.71   574.4 2640.77     591 2643.35
   600.1 2649.23   628.4 2658.81   674.1 2672.11   723.4 2684.34   790.7 2704.49
#Mann= 3 ,-1,0
       0      .1       0  419.59    .045       0   440.1      .1       0
Bank Sta=419.59,440.1
XS Rating Curve= 0 ,0
Exp/Cntr(USF)=0,0
Exp/Cntr=0.3,0.1

Type RM Length L Ch R = 1 ,75302   ,233.5,228.2,222.7
XS GIS Cut Line= 4
2263008.81153199673434.2853446132263062.19238089673828.391176804
2263083.75339695673907.8906155852263222.59242298674241.258479205
#Sta/Elev= 30
       0 2647.74    27.1 2639.49    51.4  2634.5    75.6 2627.41   128.1  2615.7
   169.1 2610.32   196.7  2603.1     229 2602.76   245.1 2606.32   321.8 2605.14
   350.1 2602.48   370.2 2597.03   415.1    2595   427.5 2592.96   435.8    2594
  443.392591.919   452.4 2590.82  459.472591.918   477.3 2594.95   490.1 2599.66
   507.5 2601.71   524.8 2608.19   581.1 2624.04   595.6 2626.79   637.2 2641.15
   732.2 2666.64   747.5 2669.01   781.2 2681.37   815.1  2689.7   841.2 2701.59
#Mann= 3 ,-1,0
       0      .1       0  443.39    .045       0  459.47      .1       0
Bank Sta=443.39,459.47
XS Rating Curve= 0 ,0
Exp/Cntr=0.3,0.1

Type RM Length L Ch R = 1 ,75074   ,217.1,226.7,237.5
XS GIS Cut Line= 4
2262850.53916709673516.6928428792262816.29402486673937.814192588
2262913.79093974674030.0053054972263035.42896406674265.983072672
#Sta/Elev= 30
       0 2643.79    60.7 2631.67    84.8 2629.97    96.8 2625.86   104.8  2625.3
   225.2 2602.97   249.3 2601.07   292.1 2595.75   313.5 2596.62   333.6 2594.99
   353.6 2589.78   365.7 2588.19   369.7 2588.76   389.8 2586.06   430.5 2587.26
   450.7 2586.21   498.4 2588.41   510.4 2588.21 515.3652586.752     521 2585.41
 540.0352586.752   543.6 2587.91   557.8 2596.87   569.7 2601.97   632.3 2615.26
   673.7  2628.8   708.8 2637.22   727.1 2643.46   774.6 2655.84   822.2 2666.04
#Mann= 3 ,-1,0
       0      .1       0 515.365    .045       0 540.035      .1       0
#XS Ineff= 2 , 0
          502.14 2597.45
Permanent Ineff=
       F       F
Bank Sta=515.365,540.035
XS Rating Curve= 0 ,0
Exp/Cntr(USF)=0,0
Exp/Cntr=0.3,0.1

Type RM Length L Ch R = 1 ,74848   ,313.2,313.7,311.3
XS GIS Cut Line= 4
 2262686.1570175673583.7800148042262700.78981848674031.834605001
2262689.71165506674103.2799871832262813.95516554674363.450839846
#Sta/Elev= 30
       0 2649.92     9.4 2648.45    21.4 2644.51    61.4 2635.31    81.4 2628.41
   101.5    2626   137.5  2619.1   162.2    2613   253.5 2597.47   269.5 2596.76
   305.6 2591.59   321.6 2586.64   334.5 2579.72   345.6 2579.74   357.6 2583.27
   377.6 2584.08   409.6 2580.63     457 2581.26  488.082579.106   495.6    2578
  505.662579.105   520.6 2581.18   531.6 2585.25   553.9 2587.09   591.3 2597.75
   620.2 2607.95   651.2 2616.44   664.9 2618.71   745.9 2637.75   808.9  2653.9
#Mann= 3 ,-1,0
       0      .1       0  488.08    .045       0  505.66      .1       0
#XS Ineff= 2 , 0
          448.28  2589.1
Permanent Ineff=
       F       F
Bank Sta=488.08,505.66
XS Rating Curve= 0 ,0
Exp/Cntr=0.3,0.1

Type RM Length L Ch R = 1 ,74534   ,207.8,208.7,205.4
XS GIS Cut Line= 4
2262489.17638703673610.1645317792262450.39157153674058.652562835
2262441.77244709674164.236837194 2262543.7654196674405.572321444
#Sta/Elev= 30
       0 2684.72    24.2 2677.31    39.2 2670.01    47.2  2668.7    66.5 2659.76
    87.3 2652.53    99.4 2645.58   115.4 2644.07   191.7 2620.79   207.8 2618.85
   243.9 2605.44     268 2603.74   284.1 2597.31   304.1  2592.6   360.4 2584.06
   396.5  2580.9   420.6 2574.61   443.5 2573.26   460.7 2569.59   494.12568.463
   504.9 2567.24  513.232568.452   520.9 2571.01     537 2569.49   558.6 2572.41
   583.2 2573.49   613.6 2585.67   674.4 2600.01   700.4  2607.8   818.1 2647.89
#Mann= 3 ,-1,0
       0      .1       0   494.1    .045       0  513.23      .1       0
#XS Ineff= 2 , 0
                          521.08         2574.74
Permanent Ineff=
       F       F
Bank Sta=494.1,513.23
XS Rating Curve= 0 ,0
Exp/Cntr(USF)=0,0
Exp/Cntr=0.3,0.1

Type RM Length L Ch R = 1 ,74325   ,222.5,224.5,224.9
XS GIS Cut Line= 4
2262309.15604038673637.7961185882262276.05102614 674006.10820259
2262257.18863685674172.7871960272262289.36880827674489.802064755
#Sta/Elev= 30
       0 2683.95    46.8 2671.06    63.6 2669.99   127.9 2652.08     148 2645.35
     160 2639.03   176.1 2637.43   208.2 2622.61   256.4 2606.56   264.4 2600.54
   268.5 2598.87   284.5 2598.15   300.6 2590.69   316.7 2585.06   352.8  2578.6
   380.9 2565.16   433.3 2561.31   477.6    2564   507.52562.815  519.772562.801
   533.9    2568   566.2 2566.86   582.2 2563.85   610.3 2565.04   630.4 2573.07
   658.6 2579.32   698.8 2590.62   803.4 2630.76   834.4 2639.97   856.2 2644.29
#Mann= 3 ,-1,0
       0      .1       0   507.5    .045       0  519.77      .1       0
#XS Ineff= 2 , 0
                          529.42         2579.52
Permanent Ineff=
       F       F
Bank Sta=507.5,519.77
XS Rating Curve= 0 ,0
Exp/Cntr=0.3,0.1

Type RM Length L Ch R = 1 ,74101   ,301.9,300,294.3
XS GIS Cut Line= 4
2262153.80434284673678.726554705 2262090.5525702 674018.09664255
2262038.24821974 674167.711412462262103.93275287674449.911628876
#Sta/Elev= 30
       0 2664.11    22.8 2663.87    59.5 2657.82    71.7 2657.14   100.1 2646.61
   112.4  2640.6   132.7 2626.94   144.9 2624.94   169.3 2612.53   201.9 2604.39
   254.8  2587.4   271.1 2586.43   283.2 2583.35   295.5 2583.75   305.3  2578.5
   332.1 2571.96   336.2 2570.07   352.7 2557.65   377.8 2555.19  392.652555.177
   416.3 2555.95   424.8 2554.01   433.2 2555.71   454.4 2556.74   479.8 2555.56
   529.9 2564.25   636.6 2574.36   706.4 2593.11   718.8 2595.41   793.5 2618.49
#Mann= 3 ,-1,0
       0      .1       0   377.8    .045       0  392.65      .1       0
Bank Sta=377.8,392.65
XS Rating Curve= 0 ,0
Exp/Cntr(USF)=0,0
Exp/Cntr=0.3,0.1

Type RM Length L Ch R = 1 ,73801   ,353.6,360.6,363
XS GIS Cut Line= 4
2261921.36888089 673758.688042552261785.14993239673986.572071197
2261837.33961076674128.7188729022261937.66303634674495.063978467
#Sta/Elev= 30
       0 2633.11    30.9 2619.58    84.9  2601.2   110.6 2590.24     166  2573.3
   175.3 2568.24   189.4 2565.89   198.6 2561.44   212.7 2559.93   226.6 2554.88
     236 2553.56   268.3 2549.25   291.7 2549.16   303.32546.955  312.792546.918
   340.7 2547.47   353.5 2544.19   372.7 2548.35   400.4 2549.05   454.7 2555.49
   504.2 2558.58   537.7 2564.88   548.8 2564.72   558.4 2566.38   605.2 2578.47
   633.1 2590.68   699.4 2614.66   740.9 2623.54   774.1  2627.7   796.8 2636.72
#Mann= 3 ,-1,0
       0      .1       0   303.3    .045       0  312.79      .1       0
Bank Sta=303.3,312.79
XS Rating Curve= 0 ,0
Exp/Cntr=0.3,0.1

Type RM Length L Ch R = 1 ,73440   ,251,246.4,239.9
XS GIS Cut Line= 4
2261827.46496705673754.8929817842261553.10364553 673937.35001826
  2261504.260484674084.7123905592261692.61576836674459.775860952
#Sta/Elev= 30
       0 2624.78    73.3 2603.23   116.5 2583.75   157.7 2569.23   170.3 2562.29
   184.7 2558.52   214.6 2544.02   293.1 2539.48   315.6 2542.53   358.8  2536.3
   378.2 2536.62   388.3 2535.08  400.672536.613     422 2539.47     494 2537.53
   520.2 2542.12   534.5 2542.38   552.4 2540.08   610.6  2544.2   642.9 2552.44
   653.9 2552.47   677.7 2558.45   696.6 2559.32     727 2572.19   740.4 2573.61
   771.7 2582.65   823.2 2600.13   843.3 2603.08   888.1 2613.67   904.4 2615.24
#Mann= 3 ,-1,0
       0      .1       0   378.2    .045       0  400.67      .1       0
#XS Ineff= 2 , 0
                           424.3         2546.05
Permanent Ineff=
       F       F
Bank Sta=378.2,400.67
XS Rating Curve= 0 ,0
Exp/Cntr(USF)=0,0
Exp/Cntr=0.3,0.1

Type RM Length L Ch R = 1 ,73194   ,400.5,397,392.3
XS GIS Cut Line= 4
2261243.83975506673768.2582166792261303.87608004673930.047767766
2261331.71139319674014.9811591752261511.10013783674502.697700509
#Sta/Elev= 30
       0  2598.1    94.8 2569.62   107.6  2563.5   116.2 2561.31   131.7 2553.62
     141 2547.44   153.5  2546.3   175.9 2535.16  197.592529.516   205.3 2527.67
  215.182529.516   243.2 2532.48   311.2 2534.44     324 2533.46   332.6  2534.4
   366.8 2531.83   432.3 2534.46   456.1 2540.94   494.6 2546.82   545.6 2556.83
   556.9 2560.43   575.4 2561.32     585 2566.94   605.2 2571.73   656.4  2588.5
   703.3 2599.64   728.3 2607.14   754.4 2612.08   762.9 2615.13   781.6 2616.88
#Mann= 3 ,-1,0
       0      .1       0  197.59    .045       0  215.18      .1       0
Bank Sta=197.59,215.18
XS Rating Curve= 0 ,0
Exp/Cntr=0.3,0.1

Type RM Length L Ch R = 1 ,72797   ,491.8,492.2,492.2
XS GIS Cut Line= 4
2260890.83068799673912.8436574132261006.43803301674208.574162356
 2261126.0310074674324.455838489 2261283.8626033674534.189051296
#Sta/Elev= 30
       0 2632.17     8.9 2627.03    17.5 2619.36    30.4 2617.53    47.6 2607.41
    56.2 2606.66    90.8 2590.29   103.2 2588.09   116.3 2582.41   143.3 2575.61
   193.6 2558.29   210.8 2549.99   223.4 2547.59   245.2 2537.94   282.3 2530.16
     356 2523.73  364.862519.881   375.8 2518.38  387.082519.879   395.6 2521.52
   449.3 2523.17   471.9 2521.73     550 2549.91   591.8 2563.09   620.1 2569.52
   634.6 2569.42   690.2 2583.24   707.1 2589.67   720.2 2591.01   746.5 2599.43
#Mann= 3 ,-1,0
       0      .1       0  364.86    .045       0  387.08      .1       0
#XS Ineff= 2 , 0
                          449.16         2528.03
Permanent Ineff=
       F       F
Bank Sta=364.86,387.08
XS Rating Curve= 0 ,0
Exp/Cntr=0.3,0.1

Type RM Length L Ch R = 1 ,72304   ,495.6,505.4,496.2
XS GIS Cut Line= 4
2260474.46501346674189.2049487042260586.86624987674459.341105926
2260741.66160238 674607.235597532260931.97869553674766.207234639
#Sta/Elev= 30
       0 2646.93    25.3 2636.72    41.1 2626.88    99.2 2598.36   126.7 2586.92
   151.6 2573.45   164.6 2571.36   229.6  2544.3   243.9 2535.64   255.2 2532.61
   276.6 2518.75   288.9 2513.13   334.4 2511.06     408 2512.77  419.172509.991
   428.4 2508.92  439.39 2509.99   449.3 2513.22   471.4 2515.32   487.2 2511.72
   498.5 2511.84   515.5 2520.71   552.4 2524.22   562.1 2527.13   588.1 2528.77
   603.3 2534.83   671.9 2553.42   711.5 2568.06   725.7  2569.6   754.7 2583.63
#Mann= 3 ,-1,0
       0      .1       0  419.17    .045       0  439.39      .1       0
#XS Ineff= 2 , 0
          398.61 2522.17  469.94         2522.89
Permanent Ineff=
       F       F
Bank Sta=419.17,439.39
XS Rating Curve= 0 ,0
Exp/Cntr=0.3,0.1

Type RM Length L Ch R = 1 ,71799   ,473.2,469.7,462.8
XS GIS Cut Line= 4
2260191.69399327674307.5972799432260246.23179273 674635.57778062
2260304.85433341674795.893359625 2260505.7998829674982.589671607
#Sta/Elev= 30
       0  2653.2    38.1 2644.24    78.6 2627.62    90.8 2624.79   123.3 2611.34
   155.7 2597.24   165.2 2590.99     180 2588.28   192.2  2579.8   236.8  2558.6
   277.3 2536.19   293.6 2532.35   317.9 2520.21   338.6 2502.74  352.962500.732
   375.8 2499.91  389.742500.727   431.9 2502.95   449.2 2501.57     462 2502.75
   481.8 2507.18   529.1 2508.08     605 2516.87     631 2524.02   673.4 2538.54
     730 2553.33   741.4 2557.75   751.9 2563.77   769.5 2564.87   777.5 2569.12
#Mann= 3 ,-1,0
       0      .1       0  352.96    .045       0  389.74      .1       0
#XS Ineff= 2 , 0
                          432.07         2511.11
Permanent Ineff=
       F       F
Bank Sta=352.96,389.74
XS Rating Curve= 0 ,0
Exp/Cntr=0.3,0.1

Type RM Length L Ch R = 1 ,71329   ,304.4,307.7,302.4
XS GIS Cut Line= 4
2259883.67915989674538.8169955592259812.43972598674817.296729567
2259935.13449528674980.7040719282260110.63194213675111.329927325
#Sta/Elev= 30
       0 2576.97    76.8 2559.05      85 2554.93   101.5  2552.6   109.8 2550.38
   167.6 2531.93   188.2  2524.2   196.5 2519.64   208.9 2517.56   241.9 2504.41
   283.2 2495.02     307 2493.96  312.842491.716   317.3 2490.62   327.3 2491.09
   337.3 2490.22  343.532491.714   357.3 2495.33   367.3 2493.71   447.4  2493.5
   457.4 2494.65   472.4 2492.32   487.2 2492.99   539.5 2506.51   562.9 2513.53
   602.8 2529.12   622.7 2533.13   652.7 2540.99   684.4  2550.6   710.6 2554.77
#Mann= 3 ,-1,0
       0      .1       0  312.84    .045       0  343.53      .1       0
#XS Ineff= 2 , 0
                          358.12         2510.47
Permanent Ineff=
       F       F
Bank Sta=312.84,343.53
XS Rating Curve= 0 ,0
Exp/Cntr=0.3,0.1

Type RM Length L Ch R = 1 ,71022   ,231.9,224.5,217.3
XS GIS Cut Line= 4
2259162.95243597674916.1263436832259565.57429646674978.161736085
2259695.80011053   675113.8826622259983.98248693 675227.66663221
#Sta/Elev= 30
       0  2619.7    21.5 2615.39      66 2602.23    78.1 2601.44   167.2 2572.76
     236  2556.9   244.1 2552.51   256.2 2552.96   280.5 2542.57   304.8 2528.72
   331.6 2518.04   359.7 2509.45   373.6 2502.34   385.7 2503.07   401.9 2491.42
   411.3 2487.75   483.6 2488.23   511.82484.771   526.7 2483.48   538.7 2484.78
   578.7 2489.42   675.4 2488.29   727.8 2495.87   761.7 2498.13   789.5 2504.73
   802.3 2511.21   829.5  2518.1   862.5 2530.25   887.6 2534.88   905.3 2540.85
#Mann= 3 ,-1,0
       0      .1       0   511.8    .045       0   538.7      .1       0
Bank Sta=511.8,538.7
XS Rating Curve= 0 ,0
Exp/Cntr(USF)=0,0
Exp/Cntr=0.3,0.1

Type RM Length L Ch R = 1 ,70797   ,237,234.5,233.1
XS GIS Cut Line= 4
2259107.50605249675119.1748936792259460.93016144675214.405080075
2259534.29721232675225.663913406 2259944.6099825675385.879947512
#Sta/Elev= 30
       0 2627.99    46.3 2610.45    58.7  2604.2    70.7 2596.17    79.4 2595.11
    91.8 2588.13   132.7 2572.55   187.1 2556.96   256.7 2542.77   290.7 2529.17
   315.7 2516.58   361.1  2485.3   369.3 2482.75   385.5 2482.15  394.752480.011
   409.6 2479.06  417.25 2480.01   434.1 2483.95   469.1 2480.62   480.9 2483.17
   502.4 2483.24   523.9 2485.88   626.9 2486.86   648.2 2490.29     657 2490.09
   672.9 2495.02   717.1 2502.15   784.1 2522.43   863.1 2543.21   880.7 2543.77
#Mann= 3 ,-1,0
       0      .1       0  394.75    .045       0  417.25      .1       0
#XS Ineff= 2 , 0
                          436.03         2492.78
Permanent Ineff=
       F       F
Bank Sta=394.75,417.25
XS Rating Curve= 0 ,0
Exp/Cntr=0.3,0.1

Type RM Length L Ch R = 1 ,70563   ,268.4,272.3,276.2
XS GIS Cut Line= 4
 2259106.8537641675249.7697567532259431.46859129675447.842612934
 2259519.4353753675448.8898365532259897.48908907675533.219336387
#Sta/Elev= 30
       0 2594.42    12.2 2592.56    29.6 2584.99   125.7 2555.79   186.8 2542.49
   256.6 2529.75   301.4 2515.01   357.7 2490.68   367.5 2487.94     385 2477.87
     397 2475.47     413 2474.23  424.642475.466     441 2474.43     461 2479.96
   482.5 2482.77   542.8 2485.22   575.6 2489.86     592 2489.58   661.6 2499.37
   698.5 2508.67   726.8 2513.73   751.8 2520.51   768.2 2523.76   784.1 2524.53
     801 2528.24   817.4 2534.16   833.8 2537.88   841.9 2541.59   855.6 2543.33
#Mann= 3 ,-1,0
       0      .1       0     397    .045       0  424.64      .1       0
Bank Sta=397,424.64
XS Rating Curve= 0 ,0
Exp/Cntr(USF)=0,0
Exp/Cntr=0.3,0.1

Type RM Length L Ch R = 1 ,70290   ,483.6,483.1,481.9
XS GIS Cut Line= 4
 2259086.9257519675422.3124852732259369.93072475675652.195516331
2259479.84174295675711.9200913072259863.82605383675835.467312851
#Sta/Elev= 30
       0 2570.97      48 2558.41    73.8 2550.16   167.9 2529.18   201.2 2519.24
   207.7 2518.35     249 2507.28   284.4 2496.68   310.8 2485.24   349.8 2472.47
   367.2 2470.27   376.3 2467.16   383.4 2466.55     399  2468.9     440 2468.81
  447.052466.985   452.5 2465.32   462.8 2466.98     490  2471.6     510 2477.05
   523.7 2479.34   554.5 2480.29   574.1 2484.38   590.9  2486.2   674.9 2508.55
   716.7 2520.72   742.2 2524.35   767.5 2530.33   876.6 2543.12   893.1 2543.86
#Mann= 3 ,-1,0
       0      .1       0  447.05    .045       0   462.8      .1       0
Bank Sta=447.05,462.8
XS Rating Curve= 0 ,0
Exp/Cntr=0.3,0.1

Type RM Length L Ch R = 1 ,69807   ,364.1,372.9,377
XS GIS Cut Line= 4
2259038.77816376675711.8845520012259106.41087972676033.202218164
 2259167.5050431676072.8332620852259584.01595356676139.029207948
#Sta/Elev= 30
       0 2521.14   115.8 2508.77   140.3 2505.02   168.9 2497.68   189.4 2493.37
   222.1 2489.85   265.7 2483.45   295.6 2475.48   307.9 2473.07   336.12459.178
     340 2457.87     347 2457.22   355.6 2457.52  362.63 2459.18     373 2461.16
   382.9 2460.98   396.1 2462.03   422.1 2460.59   515.3 2461.96   541.9 2464.97
   592.2  2467.6   628.7 2471.26   644.9 2471.94   673.2 2475.51   701.6  2480.9
   729.9 2488.02   758.3 2491.78   766.4 2493.93   782.6 2495.59   822.9 2504.55
#Mann= 3 ,-1,0
       0      .1       0   336.1    .045       0  362.63      .1       0
Bank Sta=336.1,362.63
XS Rating Curve= 0 ,0
Exp/Cntr=0.3,0.1

Type RM Length L Ch R = 1 ,69434   ,237.2,238,237.8
XS GIS Cut Line= 4
2259000.57890078675968.3065726842258923.54148538676299.432305544
2258949.22062385676596.7696983172259042.47644249676765.711398755
#Sta/Elev= 30
       0 2486.16    54.3 2479.69   103.6 2472.62   148.7 2463.12   177.2  2458.1
   193.9 2457.62   206.2 2458.87   214.5 2458.11   222.7 2459.11     231 2457.31
   271.9 2455.92   310.9 2457.11   337.7  2456.9   361.8 2456.01  384.222453.451
   393.8 2452.88  399.862453.436     410 2454.73     426  2453.3   438.1 2454.03
   482.6 2454.21   486.3 2454.13   494.3 2451.93   514.4 2451.27   526.4  2452.8
   542.5 2452.96   566.6 2455.42   626.7 2456.78   766.8 2468.78   831.4 2473.42
#Mann= 3 ,-1,0
       0      .1       0  384.22    .045       0  399.86      .1       0
Bank Sta=384.22,399.86
XS Rating Curve= 0 ,0
Exp/Cntr(USF)=0,0
Exp/Cntr=0.3,0.1

Type RM Length L Ch R = 1 ,69196   ,83.4,78.4,78
XS GIS Cut Line= 6
2258809.72207062675878.8915998342258719.55377149676152.002627976
2258731.22290471676229.3822820452258769.76410754 676502.38246872
2258786.46529543676587.8154683142258905.17446198676799.824138687
#Sta/Elev= 30
       0 2483.16    10.8 2480.97    25.2 2477.06    61.4 2475.97    82.4 2471.01
    95.1 2470.58   116.1 2466.17   145.6 2462.28   170.9 2459.44   225.7 2455.22
   296.9 2452.94   337.3 2452.53   369.7 2453.04   490.9 2451.18   616.1 2452.23
   620.2 2452.02  624.092449.637   628.2 2448.55   632.3 2448.47  640.242449.637
   648.5  2452.9   660.7 2450.69   668.9 2451.19     677 2452.88   697.4 2452.67
   764.9  2455.9   816.1 2461.01   863.1 2463.81   959.4 2474.37   971.6 2474.87
#Mann= 8 ,-1,0
       0      .1       0      30     .06       0     130     .05       0
  435.87     .06       0  624.09    .045       0  640.24     .06       0
  778.62      .1       0  958.62     .06       0
Bank Sta=624.09,640.24
XS Rating Curve= 0 ,0
Exp/Cntr=0.3,0.1

Type RM Length L Ch R = 1 ,69118   ,163.7,173.6,175.8
XS GIS Cut Line= 6
2258731.21221301675883.1739557032258641.04391388676156.284983845
2258652.71304711676233.6646379152258691.25424993676506.664824589
2258707.95543782676592.0978241842258826.66460437676804.106494556
#Sta/Elev= 30
       0 2475.21    52.7 2467.56   111.6 2460.69   128.5  2460.1     158 2456.75
   195.9  2456.3   225.4 2454.93   263.7 2451.36   300.7  2450.7   405.8 2450.83
   435.8 2449.75   486.6 2451.61   510.8 2449.35     542 2449.74   555.2 2450.77
     588 2449.72   595.6 2450.12  603.212448.904   615.8 2447.87   640.1 2447.49
  650.132448.904   656.4 2449.76   672.7 2449.65   684.9 2450.46   705.3 2453.76
   747.2 2455.63     759 2456.93   780.3 2457.27   810.9 2460.46   971.6  2473.3
#Mann= 10 ,-1,0
       0      .1       0      20     .06       0  425.87     .05       0
  531.29      .1       0  603.21    .045       0  650.13      .1       0
  728.62     .05       0  738.62     .06       0  938.62      .1       0
  958.62     .06       0
Bank Sta=603.21,650.13
XS Rating Curve= 0 ,0
Exp/Cntr=0.3,0.1

Type RM Length L Ch R = 1 ,68944   ,789.9,804.7,811.3
XS GIS Cut Line= 3
2258588.53023246675943.1548845742258499.73447471676145.074004939
 2258550.7814725676769.272847387
#Sta/Elev= 30
       0 2456.17    45.9 2452.13      94 2448.57   107.1 2448.07   133.3 2448.38
   149.9 2447.69   162.7 2447.86     190 2447.19   207.6 2446.89   228.7 2447.48
   264.8 2447.04   337.1 2447.41   362.1 2446.87   410.3 2448.69   493.6 2446.67
   509.6 2447.19   521.7 2446.55  533.282445.178   545.8 2444.48   551.3 2445.18
   558.7 2446.22   573.9 2447.28   589.9 2449.62     610 2450.06     614  2450.7
     626 2450.75   638.1  2450.2   687.9  2452.5   710.3 2454.66   846.9 2464.96
#Mann= 8 ,-1,0
       0     .05       0     190     .07       0  370.58      .1       0
  390.58     .05       0  470.58      .1       0  533.28    .045       0
   551.3      .1       0  570.58     .05       0
#XS Ineff= 2 , 0
          349.31 2450.37
Permanent Ineff=
       F       F
Bank Sta=533.28,551.3
XS Rating Curve= 0 ,0
Exp/Cntr(USF)=0,0
Exp/Cntr=0.3,0.1

Type RM Length L Ch R = 1 ,68140   ,842.5,872.2,869.5
XS GIS Cut Line= 4
2258477.78946228675708.4071554132258232.70575249676064.429618511
2258077.54196345676271.628055372     2257931.663      676634.346
#Sta/Elev= 30
       0 2468.27    15.5 2466.11    38.1 2464.48    50.6  2461.8    59.3 2462.58
    78.6 2458.24   161.2 2449.64   194.4 2448.89   272.9 2442.47   365.1  2443.2
   453.1 2441.84   479.8 2442.38   543.1 2440.73     556 2442.48   573.2 2441.53
   588.1 2441.99   599.62439.813   608.1 2438.69  621.262439.812   627.4 2441.76
   653.2 2443.63     766 2446.74     779 2448.35   830.7 2452.18   840.9 2453.93
   860.9 2453.72   873.8  2455.9   912.6 2458.63   988.5 2468.21    1082  2485.5
#Mann= 8 ,-1,0
       0      .1       0     240     .05       0     290     .07       0
  462.22      .1       0   599.6    .045       0  621.26      .1       0
  721.08     .05       0  851.08      .1       0
#XS Ineff= 2 , 0
           479.9 2446.46
Permanent Ineff=
       F       F
Bank Sta=599.6,621.26
XS Rating Curve= 0 ,0
Exp/Cntr=0.3,0.1

Type RM Length L Ch R = 1 ,67267   ,649.2,659,648.9
XS GIS Cut Line= 4
2258276.38013599675518.1444216462258023.71653399675771.906111729
2257738.34623436676052.767264939     2257554.026      676360.575
#Sta/Elev= 30
       0 2474.15   102.3 2462.36     159 2458.68   198.7 2452.02   289.4 2443.23
     377 2438.77     408 2439.29   485.4 2436.59   536.7 2438.05   570.9 2435.49
   593.7 2436.23  603.162434.448   616.1 2432.45   624.6 2432.99  628.062434.449
     633 2436.13     645 2436.07   666.1 2438.55   696.4 2436.48   727.9 2436.25
   753.4 2439.99   821.6 2443.68   880.2 2450.96   926.6 2461.01   954.8 2469.71
   964.1 2470.79   987.4 2478.22  1074.2 2500.15    1090 2505.72  1117.3 2524.79
#Mann= 3 ,-1,0
       0      .1       0  603.16    .045       0  628.06      .1       0
#XS Ineff= 2 , 0
          528.38 2443.62  663.18         2443.68
Permanent Ineff=
       F       F
Bank Sta=603.16,628.06
XS Rating Curve= 0 ,0
Exp/Cntr=0.3,0.1

Type RM Length L Ch R = 1 ,66608   ,429.5,433.7,433.5
XS GIS Cut Line= 4
 2257764.6227328675316.5059876142257586.15420037 675540.20002525
2257472.08110344675870.351318969     2257375.482      676245.133
#Sta/Elev= 30
       0 2465.81      20 2461.64    41.8 2460.17    66.3 2456.24   246.5 2438.76
     274 2434.75   371.8 2432.86     393 2434.06   422.6 2430.94   443.8 2431.91
  451.162430.698   467.8 2429.48  473.02  2430.7   507.3  2432.1   532.7 2431.11
   549.6 2431.97   566.5 2430.71   584.1 2435.13   625.8 2437.03   712.7 2447.85
   725.1 2448.56   762.3 2455.93   853.2 2477.07   894.5 2488.29     911 2489.68
     940 2499.04   968.8 2505.45   981.2 2511.24  1012.1 2529.83  1022.5 2534.49
#Mann= 3 ,-1,0
       0      .1       0  451.16    .045       0  473.02      .1       0
Bank Sta=451.16,473.02
XS Rating Curve= 0 ,0
Exp/Cntr=0.3,0.1

Type RM Length L Ch R = 1 ,66175   ,389.4,385.7,372.5
XS GIS Cut Line= 4
 2257414.4240513675303.5459223512257258.03888883675575.547186681
2257175.28677208675717.114686182 2257082.0389487676059.330631059
#Sta/Elev= 30
       0 2453.78    29.6 2451.54      48 2448.44    73.2 2447.29     108 2443.77
     168 2444.81   214.1 2439.92   292.6 2435.58   304.6 2433.44   333.3 2433.54
   348.5  2431.7  358.462427.632     362 2426.28   375.9 2425.28  388.142427.632
   415.7 2427.59     450  2430.5     511 2444.65   535.7 2447.81   578.1 2456.95
   697.5 2488.43   721.4 2493.31   734.4  2494.5   743.1 2498.32   755.6 2501.84
     764 2506.83   772.2 2509.84   805.3 2515.19   817.8 2518.53   832.4 2527.74
#Mann= 3 ,-1,0
       0      .1       0  358.46    .045       0  388.14      .1       0
Bank Sta=358.46,388.14
XS Rating Curve= 0 ,0
Exp/Cntr=0.3,0.1

Type RM Length L Ch R = 1 ,65789   ,496.5,494.5,484
XS GIS Cut Line= 4
2257047.44306056675120.126029608      2256922.97675471.113421268
2256918.90399142675603.1337222522256898.65105518675973.811969046
#Sta/Elev= 30
       0 2462.19    81.8 2451.19   128.4 2447.12   158.1 2443.36   234.5  2437.9
   336.4 2435.36   349.1 2433.08   369.9 2433.99   414.5 2430.59  432.132425.781
   446.5 2423.63   458.5  2424.5  462.632425.778   470.7 2428.69   486.5 2429.79
   497.5 2431.84     528 2440.83   554.6 2444.37   562.6  2446.4   582.6 2448.56
   594.7  2448.8   602.7 2451.56   706.8 2472.28   742.9 2476.54   766.9 2481.49
     787 2487.05     799 2492.07     827 2500.86     851 2510.29   875.7 2513.08
#Mann= 3 ,-1,0
       0      .1       0  432.13    .045       0  462.63      .1       0
Bank Sta=432.13,462.63
XS Rating Curve= 0 ,0
Exp/Cntr=0.3,0.1

Type RM Length L Ch R = 1 ,65294   ,508,499.8,490
XS GIS Cut Line= 4
2256340.31669087675043.9604617122256459.96985225675411.218988595
2256505.28385979675494.8962841982256630.45630687675905.595001132
#Sta/Elev= 30
       0 2470.34    23.1 2465.55    47.6  2464.4    64.4 2460.41    85.4 2460.16
   102.8 2454.79     178 2446.06     220 2436.66   253.7 2433.26   283.1 2427.02
   312.6 2426.22   354.7  2430.1   367.3 2428.02   384.1 2429.86   393.8 2427.23
  408.422420.257   417.4  2418.8  434.982420.258   452.2 2424.74     488 2424.17
   600.9 2433.52   613.4 2432.61   663.6 2440.26   684.3 2441.35   768.2  2456.1
   784.9 2456.95   802.8 2462.83   860.2  2473.6   881.1 2475.71   910.8 2483.21
#Mann= 3 ,-1,0
       0      .1       0  408.42    .045       0  434.98      .1       0
Bank Sta=408.42,434.98
XS Rating Curve= 0 ,0
Exp/Cntr=0.3,0.1

Type RM Length L Ch R = 1 ,64795   ,347.9,355.7,357.1
XS GIS Cut Line= 4
2255811.53581835675404.3361317642256060.85349467675588.897206414
2256163.20843367675635.1355743372256443.50902635675935.939550591
#Sta/Elev= 30
       0 2534.64    20.7 2528.16    26.8  2524.1    38.2 2522.59    55.5 2513.35
    92.6 2497.35   120.2  2482.1   150.1  2469.5   160.1 2463.38     175 2461.41
   192.7 2453.87   214.8 2441.47   239.7 2440.83   263.6 2433.41   299.4 2427.51
   307.1 2424.46  322.11  2413.9   340.1 2412.65   349.1  2413.9   379.7 2418.51
   391.5 2417.69   401.6 2420.76     465  2422.1   489.7 2425.11     600 2430.17
     644 2437.23   658.6  2437.1   687.7 2440.56   709.6 2446.64   833.7 2466.47
#Mann= 3 ,-1,0
       0      .1       0  322.11    .045       0   349.1      .1       0
Bank Sta=322.11,349.1
XS Rating Curve= 0 ,0
Exp/Cntr=0.3,0.1

Type RM Length L Ch R = 1 ,64439   ,408.3,402.6,394.3
XS GIS Cut Line= 2
2255734.61263138675661.5566668042256141.54859971676139.060736667
#Sta/Elev= 30
       0 2484.79    57.3 2461.19    71.8 2459.48     103 2450.23   125.7  2439.7
   130.9 2438.87   151.9 2439.06   162.4 2435.44   172.9 2433.53   183.4 2429.55
   224.4 2422.04     257 2417.96   278.9 2417.57   299.1  2413.7     313 2412.51
   323.1 2412.82  331.872409.413   341.3 2408.43   353.9 2409.41   360.1 2411.44
   375.4 2419.06   384.8 2421.84   406.6 2423.16   458.8  2423.7   498.8 2425.57
   545.6 2432.89   565.5 2433.91   577.6 2438.84   593.9 2442.14   627.4 2450.95
#Mann= 3 ,-1,0
       0      .1       0  331.87    .045       0   353.9      .1       0
Bank Sta=331.87,353.9
XS Rating Curve= 0 ,0
Exp/Cntr=0.3,0.1

Type RM Length L Ch R = 1 ,64036   ,273.7,270.6,271.7
XS GIS Cut Line= 4
2255404.68423212675813.2613329762255571.39157721675956.026665738
2255737.85071191676016.4671771832256069.45243182 676271.63457686
#Sta/Elev= 30
       0 2509.55    62.5 2481.74    90.4 2466.33   104.7 2464.97   135.2 2447.51
   167.9 2446.24     184 2438.05   212.3 2428.54   230.4 2417.36   245.6 2402.84
   250.1 2401.22   258.6 2401.02  270.492402.848   292.7 2403.76   309.7 2401.41
     331 2403.66     365 2402.89   386.3 2408.75   404.3 2411.51   424.4 2410.97
     450 2415.68   581.2 2420.34     587 2419.33   633.9    2423   666.7 2429.56
   677.1 2433.44   697.3 2434.31   707.4  2436.3   762.9 2451.23     815 2462.73
#Mann= 3 ,-1,0
       0      .1       0   245.6    .045       0  270.49      .1       0
Bank Sta=245.6,270.49
XS Rating Curve= 0 ,0
Exp/Cntr(USF)=0,0
Exp/Cntr=0.3,0.1

Type RM Length L Ch R = 1 ,63766   ,115.1,114.1,113
XS GIS Cut Line= 4
2255333.63117765675993.2249232872255583.10426508676202.231904038
 2255699.3724692676248.4387905312256020.62798923676400.622955587
#Sta/Elev= 30
       0 2456.61    31.1 2453.98    49.8 2447.71    60.7 2441.73     104 2428.26
   118.1 2426.46   166.5 2416.57     212 2410.43   302.8 2409.92   314.1 2405.83
   330.9 2404.72   343.8 2402.03   362.4 2397.27  371.952392.999   386.9 2391.82
  391.89    2393   411.7 2405.53   422.1 2408.39   455.9 2412.41   489.7  2411.9
   535.6  2414.9   553.8  2419.2   566.5 2420.33   615.2 2432.28   634.9 2433.93
   643.9 2438.08     659 2442.59   752.4 2461.45   792.3 2472.22     806 2478.22
#Mann= 3 ,-1,0
       0      .1       0  371.95    .045       0  391.89      .1       0
Bank Sta=371.95,391.89
XS Rating Curve= 0 ,0
Exp/Cntr=0.3,0.1

Type RM Length L Ch R = 1 ,63652   ,128.8,132,135.2
XS GIS Cut Line= 4
2255311.17432814676048.5208799222255513.35132112676305.675827132
2255631.28790035676340.2587338252255880.46217679676455.535089471
#Sta/Elev= 30
       0 2452.51      21 2444.23    61.9 2432.85    72.1 2427.92   107.7  2420.1
   137.5 2415.27     240 2404.02   274.6 2402.96   316.3 2404.26   326.5 2402.21
   346.7 2394.58   359.2 2393.63   380.6 2395.26   392.6 2393.97  401.382390.691
   405.1 2389.36   417.6 2388.97   424.9 2390.68     445 2404.93   455.4 2407.81
   468.6 2406.01   490.7 2406.31   511.6 2409.31   532.7 2410.45     592 2420.27
   609.7 2421.51   632.2 2428.68   653.7 2430.18   665.3 2435.61   724.6 2450.35
#Mann= 3 ,-1,0
       0      .1       0  401.38    .045       0   424.9      .1       0
Bank Sta=401.38,424.9
XS Rating Curve= 0 ,0
Exp/Cntr(USF)=0,0
Exp/Cntr=0.3,0.1

Type RM Length L Ch R = 1 ,63520   ,99.3,101.2,102.6
XS GIS Cut Line= 4
2255232.35866295 676092.537857882255425.84933366676380.604686024
2255554.26466669676456.9597489052255842.33149483676575.830699073
#Sta/Elev= 30
       0 2448.52    44.1 2434.93   128.8 2415.52   140.5 2413.91   159.8 2407.73
   222.1  2406.8   285.1  2400.1   300.1 2400.56   331.8 2398.84     344 2396.74
     356 2391.42   363.8 2389.31   405.6 2390.52   418.6 2392.14   449.9 2392.17
  457.722390.752     463 2389.53  467.642390.768   475.4 2393.34   515.8 2401.19
   550.1 2401.15     593 2403.54   606.7 2407.94   615.3 2408.67   671.6 2420.52
   688.9 2424.85   697.5 2428.41   719.2  2430.3   727.8 2434.72     808 2457.91
#Mann= 3 ,-1,0
       0      .1       0  457.72    .045       0  467.64      .1       0
#XS Ineff= 2 , 0
          445.97 2399.44
Permanent Ineff=
       F       F
Bank Sta=457.72,467.64
XS Rating Curve= 0 ,0
Exp/Cntr(USF)=0,0
Exp/Cntr=0.3,0.1

Type RM Length L Ch R = 1 ,63418   ,138.9,142.9,145.9
XS GIS Cut Line= 4
2255167.98916199676145.4336935232255378.34469584676426.332782968
2255500.51711097676555.9948678612255761.21902297676664.177293929
#Sta/Elev= 30
       0 2450.08    59.6 2433.69      67 2430.81    79.6 2429.55    94.6  2424.9
   105.7 2423.53   159.6 2411.84   189.6 2407.28   204.6 2403.91   249.5 2401.15
   284.5 2397.54   337.1 2396.74   344.5 2395.12   360.3 2389.44   388.6 2386.84
   404.3 2386.68   431.8 2389.04  458.34 2386.23   475.8 2384.94   481.2 2386.23
   492.9 2394.23   497.7 2395.32   587.9  2396.5   632.7 2402.07     676 2413.25
   706.3 2419.04     720 2422.97   745.3 2425.59   766.9 2432.77   811.3 2442.64
#Mann= 3 ,-1,0
       0      .1       0  458.34    .045       0   481.2      .1       0
Bank Sta=458.34,481.2
XS Rating Curve= 0 ,0
Exp/Cntr(USF)=0,0
Exp/Cntr=0.3,0.1

Type RM Length L Ch R = 1 ,63276   ,141.7,140.8,134.3
XS GIS Cut Line= 4
2255111.24903006676200.1695689172255298.47684541676500.006979471
2255355.59111488676622.2801004552255702.03875439676777.631370954
#Sta/Elev= 30
       0 2448.79    48.3 2435.34    62.4 2433.86   142.7 2412.77   152.1 2411.93
   158.2  2409.2     171 2408.61   227.5  2397.3   271.4 2390.75   281.2  2391.5
   321.9 2389.23   354.8  2389.9   376.9 2388.36   390.1 2387.15  407.622381.815
   421.9 2380.83  429.912381.814   438.7 2384.55   465.2 2383.97   478.4 2386.72
   546.1 2390.97   573.7  2389.5   611.8 2389.89     652 2393.85   681.3 2399.34
   700.8 2401.27   766.5 2417.63   787.2 2419.89   800.3 2426.13   868.1 2442.42
#Mann= 3 ,-1,0
       0      .1       0  407.62    .045       0  429.91      .1       0
#XS Ineff= 2 , 0
                          446.21         2393.77
Permanent Ineff=
       F       F
Bank Sta=407.62,429.91
XS Rating Curve= 0 ,0
Exp/Cntr=0.3,0.1

Type RM Length L Ch R = 1 ,63135   ,87.4,85.7,83.8
XS GIS Cut Line= 4
2255049.93799157676291.1882569632255195.75765512676606.474015995
2255286.40231085676698.1039397132255584.93851393676798.601275404
#Sta/Elev= 30
       0 2436.31      11 2434.86    19.8 2430.71    59.5 2416.95    81.6 2414.28
    90.6 2410.96   121.2 2404.56     193 2391.52   262.3 2383.86   291.2 2384.66
   306.3 2383.02   322.6  2383.2   341.5 2380.42   399.2 2380.76   416.2 2378.84
   423.1 2375.93   435.6 2373.79  448.092375.944   462.7  2380.1   516.1 2384.17
   609.6 2384.55   621.6 2387.61   638.5 2388.26   651.2 2391.18   666.4 2392.36
   686.5 2396.89   704.3 2398.03   765.1 2409.49   777.8 2413.86   791.3 2415.34
#Mann= 3 ,-1,0
       0      .1       0   423.1    .045       0  448.09      .1       0
Bank Sta=423.1,448.09
XS Rating Curve= 0 ,0
Exp/Cntr(USF)=0,0
Exp/Cntr=0.3,0.1

Type RM Length L Ch R = 1 ,63049   ,275,268.4,276.5
XS GIS Cut Line= 3
2254936.57750506676532.7015280122255349.97625123676843.149621174
2255575.03116709676903.802719067
#Sta/Elev= 30
       0 2405.42    34.1 2402.87    54.5 2398.32    94.1  2393.3     120 2386.75
   185.8 2380.14   217.2 2379.94   229.6  2377.8   288.6 2379.04   294.6 2378.08
  308.942372.268   322.9 2370.65   333.9 2372.26   342.9 2376.78   351.5 2377.64
   394.3 2378.52   405.7 2377.21   419.7 2379.34   437.2 2378.54   448.6 2379.79
   469.7 2379.88   494.7 2377.87     517 2378.74   577.3 2388.89   610.4 2392.65
   683.6  2404.9   693.9 2407.94     714 2408.83     726 2412.97   750.1 2418.11
#Mann= 3 ,-1,0
       0      .1       0  308.94    .045       0   333.9      .1       0
Bank Sta=308.94,333.9
XS Rating Curve= 0 ,0
Exp/Cntr(USF)=0,0
Exp/Cntr=0.3,0.1

Type RM Length L Ch R = 1 ,62781   ,252.4,248.8,249.3
XS GIS Cut Line= 3
2254791.49624961676569.2891278262255293.65260868677006.244589621
2255482.33677729676997.552171812
#Sta/Elev= 30
       0  2428.7    16.8 2422.56      38 2419.15    48.6 2414.09    59.2 2413.94
    91.2 2404.54   112.2 2400.45   130.8 2394.33   176.5 2383.03   218.7 2374.47
   260.7  2368.1   316.7 2371.04   329.3 2369.67   340.2 2371.18   431.4 2372.53
   505.6 2370.13   517.8 2367.49     547 2365.89   578.8 2366.81  584.952364.792
   589.5 2363.92   610.7 2364.79   618.5  2367.3   646.8 2367.51   703.5 2373.71
   755.3  2385.9   784.3 2388.41   833.7  2398.6   844.4 2401.35   854.5 2405.94
#Mann= 3 ,-1,0
       0      .1       0  584.95    .045       0   610.7      .1       0
#XS Ineff= 2 , 0
                          622.22          2372.2
Permanent Ineff=
       F       F
Bank Sta=584.95,610.7
XS Rating Curve= 0 ,0
Exp/Cntr(USF)=0,0
Exp/Cntr=0.3,0.1

Type RM Length L Ch R = 1 ,62532   ,290.7,304.2,317.7
XS GIS Cut Line= 4
2254712.38824898676714.4728889032255031.43480747677009.326343435
2255134.25549931677069.8091033392255441.20550582677139.364277229
#Sta/Elev= 30
       0 2433.18    24.4 2428.87    48.7 2420.85      57 2419.42    66.9 2412.54
    80.6 2410.19    92.3 2401.78   109.3 2395.58   214.1 2369.72   275.1 2359.87
   296.1 2360.07   335.8 2356.22   359.2 2360.75   375.5 2358.86     393 2352.79
   428.3 2359.68   449.9 2360.73   458.5 2360.19  471.542353.884   484.5 2352.92
  490.75 2353.86   510.8 2360.53   520.9  2362.3   563.9 2360.98     650 2362.65
   744.4 2376.89   764.9 2377.88   806.3 2385.53     851 2390.13   868.5 2394.01
#Mann= 3 ,-1,0
       0      .1       0  471.54    .045       0  490.75      .1       0
#XS Ineff= 2 , 0
          441.88 2379.35
Permanent Ineff=
       F       F
Bank Sta=471.54,490.75
XS Rating Curve= 0 ,0
Exp/Cntr(USF)=0,0
Exp/Cntr=0.3,0.1

Type RM Length L Ch R = 1 ,62228   ,219.7,202.6,184.4
XS GIS Cut Line= 4
2254638.86298789676782.6890780592254824.78844131  677058.8295651
2254806.37538004677190.3171251992255219.14405114677386.311858687
#Sta/Elev= 30
       0 2448.11      20 2439.14      46 2429.37    74.8 2415.09    83.4 2414.36
    97.8 2410.69   146.8 2392.63   181.4 2382.25   215.2 2374.99   234.5 2368.82
   253.5 2365.62   287.5 2355.29   326.1 2348.18   351.4 2339.37   359.5 2338.78
   371.6 2340.68   387.8 2341.29   407.32338.453   424.1 2337.25  434.532338.454
   440.3 2340.04   464.5 2339.67   480.9 2342.33   621.5 2345.49   649.2 2348.86
   658.3 2346.65   677.5 2345.42   721.4 2346.68   871.5 2357.91   922.6 2364.17
#Mann= 3 ,-1,0
       0      .1       0   407.3    .045       0  434.53      .1       0
Bank Sta=407.3,434.53
XS Rating Curve= 0 ,0
Exp/Cntr=0.3,0.1

Type RM Length L Ch R = 1 ,62025   ,245.4,244.8,243.3
XS GIS Cut Line= 4
2254509.06615738676909.4316588882254628.37329682677228.937581597
2254759.61099401 677267.067453082255158.64453279677420.473680209
#Sta/Elev= 30
       0 2424.74    16.8 2419.81    29.6 2418.65   101.7  2390.1   153.4    2374
     162 2373.97   187.6 2368.01   247.4 2360.31   307.2 2348.42     345 2343.97
   360.5 2338.53  368.262333.203   378.3 2330.38  390.292333.191     396 2335.69
   461.6  2334.3   478.3 2338.77   513.8 2340.42   532.4 2338.64   598.3 2339.19
   636.9 2342.77   675.5 2341.53   706.5 2342.65     744  2348.5   752.2 2345.36
   767.7 2345.22   786.9 2347.94   808.3 2347.39   872.6 2356.27   905.2 2358.31
#Mann= 3 ,-1,0
       0      .1       0  368.26    .045       0  390.29      .1       0
Bank Sta=368.26,390.29
XS Rating Curve= 0 ,0
Exp/Cntr(USF)=0,0
Exp/Cntr=0.3,0.1

Type RM Length L Ch R = 1 ,61780   ,286.2,295.2,302.9
XS GIS Cut Line= 4
2254209.60300404677270.1479609712254616.69363309677471.901769082
2254747.07810863677490.7026537162255135.56502961677590.625966354
#Sta/Elev= 30
       0 2390.94     2.9 2390.76    11.8 2384.44    20.7 2380.89   114.9  2364.3
   185.9 2357.09     205 2353.82   286.1 2347.42   319.8 2341.85   351.1 2340.59
   400.2  2335.4   413.6 2335.77     440 2331.43   465.9 2329.13   486.1 2330.03
   494.2 2328.12  506.132322.023   522.5 2321.15  532.162322.024   542.7 2326.78
   562.9 2325.13   591.3 2330.84   640.9 2332.93     681 2337.05   711.1 2335.37
   752.4 2336.69   871.5 2346.65   892.8 2350.68     934 2355.07   987.2 2365.16
#Mann= 3 ,-1,0
       0      .1       0  506.13    .045       0  532.16      .1       0
Bank Sta=506.13,532.16
XS Rating Curve= 0 ,0
Exp/Cntr=0.3,0.1

Type RM Length L Ch R = 1 ,61485   ,247.7,245.7,242.6
XS GIS Cut Line= 4
2254189.57227893677384.001185851 2254458.2548617677662.437921797
 2254573.2775872677776.2951057952254878.06627612677872.191773363
#Sta/Elev= 30
       0 2375.97    56.4 2361.26    78.6 2360.28   135.6 2354.28   155.4 2351.06
     212 2344.46   234.2  2339.9   262.9 2336.53   297.5 2334.39   332.1 2330.67
   342.1  2328.1   355.1 2327.41   376.1 2322.03   396.5 2313.58   415.7 2307.87
     427 2306.09   435.5 2307.92   455.3 2312.09   480.7  2312.1     543  2316.2
   577.3 2316.15   593.7 2317.75   644.1 2319.36   690.2 2323.67   723.7 2323.35
   748.9 2327.39     795  2331.3   811.8 2335.72   820.2 2334.75   868.3 2341.18
#Mann= 3 ,-1,0
       0      .1       0   415.7    .045       0   435.5      .1       0
Bank Sta=415.7,435.5
XS Rating Curve= 0 ,0
Exp/Cntr(USF)=0,0
Exp/Cntr=0.3,0.1

Type RM Length L Ch R = 1 ,61240   ,255.4,260.6,265
XS GIS Cut Line= 4
2254119.66957081677517.7963758752254262.32828672677823.553971135
2254396.28465601677921.667919527  2254815.905448678051.427841883
#Sta/Elev= 30
       0 2365.68     8.9 2364.13    20.1 2359.44      39 2355.91    74.4    2355
   190.4 2346.02   318.9 2330.26   339.7  2323.7   349.6 2316.47   359.9  2314.2
  377.582303.749   384.3 2302.48  409.842303.749     462 2308.01   498.4 2306.18
   515.9  2307.5   528.5 2311.37   553.6 2309.44   620.6 2313.15   646.9  2316.2
   691.6 2317.65   729.4 2323.53   750.4 2323.05   790.8  2326.9   800.6 2329.98
   845.1 2332.14   880.1 2339.99   896.9 2338.72   917.8 2342.15   942.7 2343.83
#Mann= 3 ,-1,0
       0      .1       0  377.58    .045       0  409.84      .1       0
Bank Sta=377.58,409.84
XS Rating Curve= 0 ,0
Exp/Cntr=0.3,0.1

Type RM Length L Ch R = 1 ,60979   ,557.9,535.1,502
XS GIS Cut Line= 4
2254045.29456469677824.0823873032254086.08465976677989.016249994
2254175.64552069678113.160017611 2254559.6044591678114.933500005
#Sta/Elev= 30
       0 2330.93    56.1 2322.28   108.3 2316.16   173.5 2303.64   185.8 2302.24
   197.3 2303.11   208.8 2299.32   214.5 2298.59  236.232299.312   243.1 2300.84
   258.9 2302.02     317 2300.84   375.3 2302.13   391.5 2300.45     436 2299.82
   494.7 2304.26   518.6 2303.32   539.5 2304.69   551.5 2303.38   559.5 2304.87
   571.5 2301.25   575.5 2301.04   587.5 2305.33   612.8 2308.98   623.5  2311.5
   651.5 2311.88   671.5 2313.18   679.5  2314.8   695.5 2313.84   706.9 2315.44
#Mann= 3 ,-1,0
       0      .1       0   208.8    .045       0  236.23      .1       0
#XS Ineff= 2 , 0
                          259.73         2308.56
Permanent Ineff=
       F       F
Bank Sta=208.8,236.23
XS Rating Curve= 0 ,0
Exp/Cntr(USF)=0,0
Exp/Cntr=0.3,0.1

Type RM Length L Ch R = 1 ,60444   ,294.7,298.2,302.9
XS GIS Cut Line= 4
2253830.19632931678442.9095108332254180.54777634678307.238107652
2254218.05692899678193.1145155642254724.82952322678154.009228765
#Sta/Elev= 30
       0 2357.82    49.3 2350.68    62.2 2346.65    86.4 2345.49     178 2328.61
   220.9 2315.49   315.3 2297.71   339.9 2296.02   407.3 2295.99  431.45 2293.39
   437.2 2292.19   453.7 2293.38   462.1    2297   478.4 2298.38   538.1 2296.61
   562.1 2299.98   594.6 2299.04   666.5 2302.72     684 2299.79   702.5 2301.71
   728.7 2301.06   743.6  2303.7     759 2302.87   793.8 2310.85   814.9 2312.11
   826.9 2316.19   870.2  2324.9   943.3 2333.34   987.4 2334.41  1004.1 2337.64
#Mann= 3 ,-1,0
       0      .1       0  431.45    .045       0   453.7      .1       0
Bank Sta=431.45,453.7
XS Rating Curve= 0 ,0
Exp/Cntr(USF)=0,0
Exp/Cntr=0.3,0.1

Type RM Length L Ch R = 1 ,60146   ,390.4,416.4,424.6
XS GIS Cut Line= 4
2253934.55298654678637.1512346382254336.84499097678484.632749873
 2254406.7533022678416.7843699172254624.44997055678302.274304468
#Sta/Elev= 30
       0  2352.3    75.7 2337.48   131.5 2330.02     160 2323.53     178 2323.58
     237 2310.49   279.8 2308.77   314.5 2304.35   335.4 2303.08   348.2 2298.62
   370.4 2300.52   403.8 2297.14     420 2296.84   452.4 2291.12  472.122290.796
   501.8 2288.94  512.632290.797   525.6 2292.79   547.3 2293.37   581.7  2291.7
   642.2  2312.2   655.8 2315.37   682.9 2324.15   705.5 2327.17   719.1 2326.22
   732.6 2329.93   746.2 2332.01   755.2 2329.87   768.8 2333.42   773.6 2332.96
#Mann= 3 ,-1,0
       0      .1       0  472.12    .045       0  512.63      .1       0
#XS Ineff= 2 , 0
                          546.43         2311.36
Permanent Ineff=
       F       F
Bank Sta=472.12,512.63
XS Rating Curve= 0 ,0
Exp/Cntr=0.3,0.1

Type RM Length L Ch R = 1 ,59729   ,230.5,225.7,221.9
XS GIS Cut Line= 4
2254024.89377255678823.0812214392254421.74043857678813.639293003
2254541.80832345678825.0573069582254825.92992183678747.290221439
#Sta/Elev= 30
       0 2346.83    67.3 2331.11    83.3 2330.09   159.3 2315.56   171.3 2312.24
   226.8 2307.44   235.3 2304.35   275.4 2300.23   287.4 2300.43   299.4  2297.3
   315.4 2297.79   343.4 2295.26   383.4 2294.71   394.9  2291.5   411.5 2283.92
  423.492281.842   443.6 2280.73  455.08 2281.84   475.8 2285.51   536.6 2291.63
   544.9 2294.59   573.9 2299.57   615.4 2310.74   644.4 2316.93     705 2323.56
   735.7  2328.8   740.8 2331.19   770.1 2331.51   781.3 2334.96   812.1 2339.75
#Mann= 3 ,-1,0
       0      .1       0  423.49    .045       0  455.08      .1       0
Bank Sta=423.49,455.08
XS Rating Curve= 0 ,0
Exp/Cntr=0.3,0.1
