HEC-RAS study ROARCK.prj: ROARCK

--- ROARCK.g01 (geometry) --- (continued)

Type RM Length L Ch R = 1 ,37678   ,426.6,413.3,407.3
XS GIS Cut Line= 4
2260459.53996051686218.5345824312260620.22260006 686258.97969817
2260968.51634334686114.9121269762261115.83693632 686052.14421761
#Sta/Elev= 30
       0 2239.64    87.3 2237.19     112 2235.54   124.6 2234.08   161.5 2227.64
   206.8 2221.55   231.3 2218.77   255.8 2216.71   308.5 2216.79   337.8 2215.18
   356.1 2214.63371.35912215.188   377.7 2215.19   386.4 2214.43   390.6 2214.69
   395.1    2216     408 2217.72     421 2220.55   433.4 2221.64     447 2224.54
   468.7 2230.44   473.2 2232.13   482.4 2234.27   494.6 2236.65   511.9 2238.91
   537.5  2240.8     564 2241.09   598.5 2243.74   649.1 2246.32   702.7  2250.7
#Mann= 5 ,-1,0
       0     .06       0      70      .1       0   337.8    .045       0
371.3591      .1       0  662.61     .05       0
Bank Sta=337.8,371.3591
XS Rating Curve= 0 ,0
Exp/Cntr=0.3,0.1

Type RM Length L Ch R = 1 ,37265   ,369.6,355.7,324.4
XS GIS Cut Line= 4
2260395.67838674686619.4493127912260636.19985942686608.815619807
 2260982.2701304686549.6753875442261286.42419337686277.536386744
#Sta/Elev= 30
       0 2258.56    84.6 2252.67   121.5 2246.82   136.6  2245.3   159.9 2240.24
   208.7 2235.91   252.9 2225.92   313.8 2216.99   346.2 2214.78   374.6 2215.66
   382.8 2214.22   419.3 2215.38   431.5 2216.92   463.9 2217.02   500.4 2218.24
   549.1 2223.81   585.7 2225.91   599.2 2228.64   604.9 2226.27   610.5 2222.68
   615.9 2221.28   621.2 2221.21   626.6  2222.1   637.3 2227.73   640.6 2228.69
   678.5 2227.99   760.7 2230.27   871.2 2235.93   952.5 2242.33    1000 2246.97
#Mann= 5 ,-1,0
       0     .05       0     190      .1       0   313.8    .045       0
   431.5      .1       0  721.84     .05       0
Bank Sta=313.8,431.5
XS Rating Curve= 0 ,0
Exp/Cntr=0.3,0.1

Type RM Length L Ch R = 1 ,36909   ,828.2,823,761.2
XS GIS Cut Line= 4
 2260507.1798751 687035.003200492260744.87972413686984.360441618
2261087.45968884686718.067915945     2261330.029      686292.911
#Sta/Elev= 30
       0 2331.93    29.6 2318.38    63.1 2300.18    78.7 2290.55      91 2279.37
   103.5 2271.04     136 2268.19   148.2 2261.63   197.3 2245.72   234.1 2235.36
   287.6 2224.28   304.7 2217.54   318.1 2213.15   338.4 2212.99   358.7 2215.84
   381.6 2214.71   395.9 2217.16   444.3 2217.81   470.1 2215.91   541.1  2219.8
   686.9 2223.61   696.4 2221.08   710.4 2220.66   737.8  2224.6   848.4 2229.15
   963.5  2230.4  1003.6 2232.97  1060.2  2241.3  1147.3 2249.48  1166.4 2249.61
#Mann= 6 ,-1,0
       0      .1       0  293.03     .12       0   304.7    .045       0
   395.9     .12       0  413.03      .1       0  846.94     .05       0
Bank Sta=304.7,395.9
XS Rating Curve= 0 ,0
Exp/Cntr=0.3,0.1

Type RM Length L Ch R = 1 ,36086   ,407.3,407.7,398.9
XS GIS Cut Line= 3
2261341.89231269687227.0933316952261339.00736941686994.318251644
2261674.98208973686615.712254766
#Sta/Elev= 30
       0  2268.5    37.9 2264.09    61.9 2260.41    69.9 2258.97   125.9  2244.9
   149.9 2240.04   177.9 2234.65   213.9 2230.23   250.4 2226.88   294.8 2224.26
   310.9 2220.56   327.9  2221.1   361.9 2218.39   415.3 2216.58   464.3 2217.06
   475.6 2214.92     491 2213.16   497.9 2212.93   511.8 2212.06  542.172212.921
   544.5 2213.74   546.1 2214.93   554.6 2222.57   560.5 2226.72   592.6 2239.93
   635.4 2253.97   662.1 2263.39   688.9 2270.88   718.9 2284.03     739  2288.6
#Mann= 3 ,-1,0
       0      .1       0   497.9    .045       0  542.17      .1       0
Bank Sta=497.9,542.17
XS Rating Curve= 0 ,0
Exp/Cntr=0.3,0.1

Type RM Length L Ch R = 1 ,35678   ,371.5,360.5,347.7
XS GIS Cut Line= 4
2261435.85058295687350.9686192512261653.12872198687204.041536302
2261834.26434685687012.091583785 2261850.8944407686816.491159561
#Sta/Elev= 30
       0 2295.85      13 2295.13    24.5 2292.88    31.8 2289.57    48.7 2278.37
    53.5 2276.09    90.8 2269.03   108.1 2264.57   111.5 2263.33   125.9 2252.19
   159.7 2242.56   212.9 2236.42   256.3  2227.4   306.1 2219.94     325 2219.63
  339.392214.439   348.7 2212.39   359.8 2211.88   400.8 2212.06   420.2 2214.42
   436.7 2212.66   456.1 2214.44   470.2 2214.43   492.8 2219.54   581.3 2234.31
   617.5 2244.35   628.2 2248.72   649.6  2255.1   693.5 2262.66   722.5 2270.31
#Mann= 3 ,-1,0
       0      .1       0  339.39    .045       0   420.2      .1       0
Bank Sta=339.39,420.2
XS Rating Curve= 0 ,0
Exp/Cntr=0.3,0.1

Type RM Length L Ch R = 1 ,35318   ,368.4,370,373.6
XS GIS Cut Line= 4
2261792.38823673687644.8000901392261974.92466537687432.766513443
2262085.57699694687208.2439027392262121.37128389687034.740006737
#Sta/Elev= 30
       0 2282.03    22.3  2280.3    67.1 2274.29    79.4 2271.62   110.3  2262.8
   155.6 2253.84   189.5 2245.29   205.3 2243.76     235 2238.68   301.3 2219.23
   310.5 2218.16   328.4 2219.56   332.8 2218.77   343.1 2213.83   352.1 2215.25
   391.2 2215.08   400.2 2213.48   453.2 2212.17  466.172215.066   471.6 2217.14
   484.5 2219.16   515.7 2227.66   548.4  2239.4   557.7 2243.42   561.6 2245.95
     570 2254.03   574.1 2256.48   590.4 2261.65   614.9 2265.27   707.2  2269.2
#Mann= 3 ,-1,0
       0      .1       0   391.2    .045       0  466.17      .1       0
Bank Sta=391.2,466.17
XS Rating Curve= 0 ,0
Exp/Cntr=0.3,0.1

Type RM Length L Ch R = 1 ,34948   ,324.7,355.6,379.1
XS GIS Cut Line= 4
2262098.10781333687767.6323278162262279.13217297687632.714269995
2262388.27243555687402.1433833022262430.11499848687239.223970283
#Sta/Elev= 30
       0 2279.05    57.5 2276.56   100.4 2267.89   123.3 2266.08   131.9 2266.75
   142.3 2264.61   194.7 2260.24   214.8 2257.37   220.5 2255.47   247.4 2241.94
   262.2 2233.51   273.9 2228.08   289.3 2221.64   304.3 2219.18  312.172214.834
   318.2 2212.93   340.2 2212.25   353.6 2212.59   362.4 2214.82   366.9 2214.95
   380.1 2212.53   397.9 2214.91   421.4 2215.42   460.5  2221.1   494.3  2229.2
   568.6 2252.98   593.4 2264.36   609.7 2273.27     636 2276.74   649.1 2277.56
#Mann= 3 ,-1,0
       0      .1       0  312.17    .045       0   362.4      .1       0
Bank Sta=312.17,362.4
XS Rating Curve= 0 ,0
Exp/Cntr=0.3,0.1

Type RM Length L Ch R = 1 ,34592   ,362.1,406.7,441.4
XS GIS Cut Line= 4
2262268.01519721 687804.918889072262524.85565382687749.901140578
2262696.18132004687637.9491211012262773.11534977687529.776464534
#Sta/Elev= 30
       0 2253.72    12.4 2252.16    28.8 2251.47    61.5 2251.79    94.2 2251.09
   106.5 2249.86   118.8  2250.3   159.7 2243.08   212.9 2231.53   229.6 2229.08
   252.6 2224.12   265.6 2219.62     281  2219.7   315.2  2216.8   332.1 2216.92
   352.6 2218.19   361.12215.077   366.7 2212.85   381.3 2210.68   395.7 2211.53
     410 2210.54   433.2 2211.28   443.4  2210.6   450.9 2212.72  455.112215.077
   462.5 2220.18     483 2229.36   494.9 2235.89   546.8 2255.85   600.1 2273.73
#Mann= 3 ,-1,0
       0      .1       0   361.1    .045       0  455.11      .1       0
Bank Sta=361.1,455.11
XS Rating Curve= 0 ,0
Exp/Cntr=0.3,0.1

Type RM Length L Ch R = 1 ,34186   ,586.9,519.3,440.7
XS GIS Cut Line= 4
 2262238.6276578687935.5643081662262484.89470701688008.623000736
2262705.42986386688076.7764139852262884.08509839687797.518897897
#Sta/Elev= 30
       0 2246.38    43.3 2244.93    66.9 2241.42    76.6 2240.83   124.8  2224.5
   172.7 2217.21   189.4 2216.18   214.4 2216.76   264.5 2219.94   293.8 2218.83
   352.4 2214.44   365.5  2214.9   394.3 2210.34   419.4 2210.05   427.8 2210.44
   434.9 2212.23  441.272214.914   457.1 2220.91   515.7 2226.79   520.5 2226.66
   532.8  2220.5   544.8  2217.5   552.2 2218.75   563.2 2225.71   567.9 2226.67
   620.2 2226.83   700.9 2224.76   752.6 2227.15   791.1 2227.91   819.2 2227.18
#Mann= 3 ,-1,0
       0      .1       0   365.5    .045       0  441.27      .1       0
Bank Sta=365.5,441.27
XS Rating Curve= 0 ,0
Exp/Cntr=0.3,0.1

Type RM Length L Ch R = 1 ,33666   ,372.3,369.8,378.8
XS GIS Cut Line= 4
2262648.39098767688709.0722758142262623.00205081688507.192208854
 2262576.8397242688264.4614111982262841.06953547687927.574135581
#Sta/Elev= 30
       0 2248.11      20 2245.37    76.5    2233   128.9 2225.22   193.4  2220.5
   213.7 2217.78   229.9 2217.82   266.6 2212.17   295.1 2212.89   339.9 2209.93
   356.2 2210.77  364.852212.879   372.5 2216.54   380.6 2217.46   396.9 2216.16
   417.2 2218.58   488.4 2220.21   515.1 2217.85   603.4 2217.71   658.1 2220.84
   689.3 2224.61   698.7 2223.16   708.9 2223.56   723.1 2218.08   734.3 2217.32
   739.4 2218.73   749.6 2224.79   771.5    2227   842.7 2226.18   878.7 2223.73
#Mann= 5 ,-1,0
       0      .1       0  223.47     .12       0   295.1    .045       0
  364.85     .12       0  570.55      .1       0
Bank Sta=295.1,364.85
XS Rating Curve= 0 ,0
Exp/Cntr=0.3,0.1

Type RM Length L Ch R = 1 ,33296   ,402.4,395.6,388
XS GIS Cut Line= 4
2262933.96442235688595.0188668842262926.00258066688328.899540798
2262952.01324662688140.9542161952263093.39585209687980.511433035
#Sta/Elev= 30
       0 2251.73    15.2  2248.5    25.9 2247.71    77.9 2238.55   105.9 2235.36
   113.9 2235.31   125.9 2232.25   133.9 2232.29   197.9 2221.22   225.9 2218.63
   278.1 2216.29   294.2 2214.23   306.3 2214.25   324.3 2212.49   350.8 2209.86
  370.322212.486   387.1 2213.11   415.4  2216.1   443.6 2216.97   466.3 2216.49
   482.3 2221.23     493  2222.8   514.3 2221.93     525 2219.14     575 2218.58
   578.3 2219.34   594.8 2227.95     621 2238.13   637.7 2241.05   669.8 2244.11
#Mann= 6 ,-1,0
       0      .1       0   324.3    .045       0  370.32      .1       0
  396.24     .12       0  515.98     .06       0  645.98      .1       0
#XS Ineff= 2 , 0
                          444.19         2224.68
Permanent Ineff=
       F       F
Bank Sta=324.3,370.32
XS Rating Curve= 0 ,0
Exp/Cntr=0.3,0.1

Type RM Length L Ch R = 1 ,32901   ,481,467.6,449.7
XS GIS Cut Line= 4
2263368.53705315688543.0764697682263336.02000985688344.253075953
2263286.99529862688102.1161743712263257.98897808687993.575181848
#Sta/Elev= 30
       0 2279.69    22.2 2272.95    50.6 2262.01      83 2254.78    99.5 2245.25
   111.4 2243.58   172.2 2229.36   216.8 2212.06  224.18 2207.49   229.1  2205.9
   249.5 2205.35  266.522207.492   294.4 2211.38   351.5 2208.52     376 2212.18
   380.1 2212.19   388.3 2210.15   404.6  2212.9     425 2210.94   429.1 2211.78
   438.1 2217.16   445.4  2219.2     466 2221.36   482.6 2221.28   486.7 2222.18
   490.9  2226.3     495 2228.83   507.5 2231.91   533.3 2241.29   560.9 2248.61
#Mann= 5 ,-1,0
       0      .1       0  224.18    .045       0  266.52      .1       0
  448.51     .06       0  558.51      .1       0
#XS Ineff= 2 , 0
                          374.91         2222.18
Permanent Ineff=
       F       F
Bank Sta=224.18,266.52
XS Rating Curve= 0 ,0
Exp/Cntr=0.3,0.1

Type RM Length L Ch R = 1 ,32433   ,62.1,63.1,70.5
XS GIS Cut Line= 6
2263859.24086493688549.5719944152263934.42150614688280.378800396
2263740.45446158688119.6074580872263679.92112217688103.335055019
2263539.97845578688104.6368472652263539.27531251688016.838808867
#Sta/Elev= 30
       0 2260.32      17 2260.08    46.1 2250.22    88.7 2238.06   133.3 2228.24
   173.1 2217.65   199.8 2215.05   212.2 2210.97   228.8 2210.85   253.7 2205.11
   307.1  2207.1   323.2 2207.29   342.8 2205.18   460.3 2207.85   466.8 2207.63
  474.472205.396   483.8 2203.96   517.6  2203.5   529.1 2205.36     535 2206.87
   552.7 2207.51     579 2203.85   603.4  2208.4   623.4 2209.44   735.6 2209.13
   743.1 2213.71   747.1 2214.83   787.1 2216.08   815.1 2231.13   823.4 2231.24
#Mann= 10 ,-1,0
       0      .1       0     260     .06       0  413.76      .1       0
  423.76     .06       0  474.47    .045       0   529.1     .06       0
  552.89      .1       0  605.66     .06       0  674.48      .1       0
  745.63     .06       0
Bank Sta=474.47,529.1
XS Rating Curve= 0 ,0
Exp/Cntr=0.3,0.1

Type RM Length L Ch R = 1 ,32370   ,554.6,577.8,590.9
XS GIS Cut Line= 6
2263889.51942522688500.5375211722263964.70006643688231.344327153
2263770.73302187688070.5729848442263710.19968245688054.300581776
2263570.25701607688055.602374022 2263569.5538728687967.804335624
#Sta/Elev= 30
       0 2246.25    20.1 2240.32    79.5 2227.24      99 2221.69   136.4 2216.32
   157.2 2210.98   173.8 2210.24   194.5 2205.01   231.9 2206.86   248.5 2205.21
   269.3 2205.49   279.5 2207.91   340.6 2208.48   358.7 2206.34   405.4 2210.18
   419.6 2209.15   433.7 2206.15     445 2204.05   476.2 2206.15   549.5 2209.44
   634.3 2207.49   677.7 2209.02     738 2213.21     742 2214.91   750.1 2223.08
   754.1 2225.36   766.1  2228.2   774.1 2232.15   795.7 2233.96   823.4 2242.96
#Mann= 5 ,-1,0
       0      .1       0     210     .06       0   433.7    .045       0
   476.2     .06       0  795.63      .1       0
Bank Sta=433.7,476.2
XS Rating Curve= 0 ,0
Exp/Cntr=0.3,0.1

Type RM Length L Ch R = 1 ,31792   ,419.9,419.6,412.9
XS GIS Cut Line= 4
 2264154.8021077688663.4180810412264262.84581443688440.166039458
2264315.20139669688181.1786900632264312.94512805688011.611829745
#Sta/Elev= 30
       0 2242.85      38 2236.35    46.9  2232.3    55.8 2230.08    82.5 2230.09
    95.5 2226.28   113.3 2222.71   168.4 2218.92   182.4 2214.03   233.3 2212.13
   255.2 2208.93   279.6 2208.96   287.8 2207.25   344.9 2201.87   353.1 2200.22
   369.4 2199.52   393.9 2201.84   402.1  2202.7   418.4 2200.44   438.8 2201.89
   471.4 2206.33   495.9  2207.5   524.2 2211.99   548.3 2219.14   588.3 2228.98
   612.3 2236.45   624.3 2241.34   640.3 2242.66   652.3 2248.77   681.8 2259.76
#Mann= 5 ,-1,0
       0      .1       0     190     .06       0  298.02      .1       0
   344.9    .045       0   393.9      .1       0
Bank Sta=344.9,393.9
XS Rating Curve= 0 ,0
Exp/Cntr=0.3,0.1

Type RM Length L Ch R = 1 ,31373   ,623.9,657.7,686.5
XS GIS Cut Line= 4
2264637.19225131688835.5666894632264665.98984149 688541.63472204
2264701.11842943688234.7834122472264607.00590672687982.726417054
#Sta/Elev= 30
       0 2272.62    18.5 2267.39    39.4 2258.97    66.7 2249.99   163.2 2227.41
   251.6 2212.37   271.7 2208.16   279.7 2204.99   295.8 2205.74     320 2203.73
   336.1 2203.67  343.03 2200.23   348.1 2197.25   356.2 2196.38  402.342200.229
   412.6 2201.61   432.7 2200.67   448.8 2202.34     481 2201.35   541.4 2202.62
   674.2 2209.99   690.1 2209.75   704.1 2211.92   721.2 2212.16   746.8 2222.26
   772.4 2234.96   789.6 2240.93   805.1 2243.46   836.5 2252.32   873.2 2266.09
#Mann= 4 ,-1,0
       0      .1       0     250     .06       0  343.03    .045       0
  402.34      .1       0
Bank Sta=343.03,402.34
XS Rating Curve= 0 ,0
Exp/Cntr=0.3,0.1

Type RM Length L Ch R = 1 ,30715   ,522.1,540.3,557.9
XS GIS Cut Line= 4
2264934.76241306688932.8254820542265115.03999535688681.713277849
 2265360.9069347688517.0963531172265594.43385922688345.438068068
#Sta/Elev= 30
       0 2274.97    43.6 2258.95    69.6 2254.55    78.3    2252    93.1 2251.89
   122.7 2245.71   147.3 2239.33   226.1 2223.12   228.8 2222.26   235.8 2216.56
   240.8 2215.08   275.9 2214.35     296 2208.42   338.8 2201.27   353.6 2201.42
   368.3  2197.8   448.7 2200.29   488.6 2198.88  507.882197.183   536.7 2194.08
   568.9 2194.46   581.82197.184   595.8  2205.9   638.9 2215.87   699.4 2236.75
   713.3 2243.62   730.3 2244.76   739.9 2249.02   793.3 2264.74   894.8 2302.56
#Mann= 5 ,-1,0
       0      .1       0     180     .06       0     300      .1       0
  507.88    .045       0   581.8      .1       0
Bank Sta=507.88,581.8
XS Rating Curve= 0 ,0
Exp/Cntr=0.3,0.1

Type RM Length L Ch R = 1 ,30175   ,485.5,484.7,464.2
XS GIS Cut Line= 3
     2265025.338      689097.8042265554.99644923689047.009827413
 2265877.7891469688988.856263824
#Sta/Elev= 30
       0 2285.82    51.1 2265.71   104.7 2254.03   127.4 2244.78   135.5 2238.37
   139.5 2237.07   155.5 2236.15   175.6 2225.72   215.8 2208.35     252  2197.8
   280.1 2195.69   320.3 2196.56   356.5 2194.52   440.9 2197.33   450.32194.762
   456.9 2192.55     473  2191.9   517.2 2193.58  521.932194.694   529.3 2199.94
   541.4 2211.12   602.4 2232.91     639 2242.06     700 2259.61   708.1 2262.93
   724.3 2264.65     765 2278.94   817.8 2293.98   838.1 2301.49   860.1 2311.65
#Mann= 5 ,-1,0
       0      .1       0     110     .06       0     190      .1       0
   450.3    .045       0  521.93      .1       0
Bank Sta=450.3,521.93
XS Rating Curve= 0 ,0
Exp/Cntr=0.3,0.1

Type RM Length L Ch R = 1 ,29690   ,440.8,446.5,443.5
XS GIS Cut Line= 4
2265046.46500633689571.0531895342265328.42888191  689532.2777933
2265591.87503186689466.885004913     2265902.905689400.743042635
#Sta/Elev= 30
       0 2301.63    42.1 2292.93    70.4 2284.79     139 2255.32   151.1 2253.77
     170 2247.24   191.5 2234.71   199.6 2227.28   219.8 2227.19   239.9  2216.4
   317.3 2196.08  333.092194.616   343.1 2192.17   392.6 2193.45   412.1  2191.8
   424.5  2194.6   473.9 2194.76   494.5 2192.91   504.8 2193.85   638.2 2222.48
   691.3 2236.32   711.8 2239.53   726.4 2244.21   748.6 2254.17   760.8 2255.56
   776.9 2264.45   814.3 2277.48   851.1 2293.33   861.3 2295.01     874 2302.34
#Mann= 5 ,-1,0
       0      .1       0     170     .06       0     270      .1       0
  333.09    .045       0   424.5      .1       0
Bank Sta=333.09,424.5
XS Rating Curve= 0 ,0
Exp/Cntr=0.3,0.1

Type RM Length L Ch R = 1 ,29243   ,389,420.1,450
XS GIS Cut Line= 4
2265162.80503552689961.1955854572265423.26382407689954.516999163
 2265712.6176273689894.2652911742265985.98872336689816.269240283
#Sta/Elev= 30
       0 2294.02     9.4 2289.95    17.4 2272.54    97.4 2240.85   109.4 2239.57
   149.4 2230.54   157.4 2224.46   181.4  2223.5   197.4  2216.1   269.6 2197.01
   306.4 2194.09   318.7 2195.24   326.8 2193.78   347.3 2194.46  352.642193.013
   416.7 2191.75   433.1 2192.98   469.9 2192.23   510.7 2194.58   539.7 2205.93
   568.1 2212.94   584.8 2215.18   622.2 2216.37   630.5 2218.16     668 2236.86
   680.4 2245.96   717.9 2258.09   767.8 2279.64   792.7 2289.01   840.4 2303.74
#Mann= 5 ,-1,0
       0      .1       0     150     .06       0     240      .1       0
  352.64    .045       0   433.1      .1       0
Bank Sta=352.64,433.1
XS Rating Curve= 0 ,0
Exp/Cntr=0.3,0.1

Type RM Length L Ch R = 1 ,28823   ,419.6,400.6,367.2
XS GIS Cut Line= 4
2265181.65536583690109.3390561842265437.30797001690259.278433655
2265597.96688639690382.0410418522265830.51566246690588.961656022
#Sta/Elev= 30
       0 2266.13    35.4 2254.52    45.6 2248.95    58.6 2246.51    86.5  2236.7
   114.2 2230.63   127.4 2224.21   151.3 2223.79   165.2 2218.47   188.8 2211.89
   197.3 2208.06   203.4 2206.67   241.4  2201.9   253.3  2198.9   267.2 2198.49
   295.1 2194.35   320.1 2194.88   340.3 2192.46   355.4 2192.19   370.5 2191.19
   420.8 2192.21   499.5 2191.83   575.5 2193.17   671.8 2197.51   689.8 2199.41
   713.9 2198.82   737.5  2200.8     756 2200.15   786.1 2201.11   809.9 2204.46
#Mann= 5 ,-1,0
       0      .1       0      30     .06       0     150      .1       0
   355.4    .045       0   420.8      .1       0
Bank Sta=355.4,420.8
XS Rating Curve= 0 ,0
Exp/Cntr=0.3,0.1

Type RM Length L Ch R = 1 ,28423   ,265.5,264.2,260.7
XS GIS Cut Line= 4
 2265022.1863191690603.1000094762265262.13488932690695.223121257
2265522.43624005690587.032024863 2265794.5207795690695.223121257
#Sta/Elev= 30
       0 2239.49      15 2234.86      45 2228.21    53.5 2220.91      75 2221.31
    86.7 2215.19   105.3 2208.33   139.7 2200.19   164.9 2198.08   254.9  2194.3
   284.6 2190.84   302.6 2190.73  348.032182.521   367.5 2180.07   393.5 2182.51
   402.2  2181.9   423.8 2187.06   467.2 2185.89   484.5 2188.38   596.7 2195.23
   652.7 2193.95   674.6 2195.33   704.4 2194.94   726.7 2196.33   747.4 2196.14
   803.4 2201.22     812 2205.61   815.4 2206.32   824.9 2204.48   831.7 2205.75
#Mann= 4 ,-1,0
       0     .06       0     170      .1       0  348.03    .045       0
   393.5      .1       0
Bank Sta=348.03,393.5
XS Rating Curve= 0 ,0
Exp/Cntr(USF)=0,0
Exp/Cntr=0.3,0.1

Type RM Length L Ch R = 1 ,28159   ,473.2,484.9,496.4
XS GIS Cut Line= 4
2264937.14574309690963.6223856332265479.06885003690891.749951724
2265596.52789883 690821.602723082265885.21068088690792.457067959
#Sta/Elev= 30
       0 2226.92    15.2 2224.26    47.4 2220.53    79.7 2213.23   104.6 2211.88
   120.1  2209.3   216.9 2197.61   261.4 2195.25   301.6  2191.2   394.5 2188.26
   402.5 2188.85   414.6 2187.03   496.5 2183.96   542.8  2181.3   557.3 2178.08
  582.592181.306   606.3 2185.21   633.9 2185.14   671.9 2189.77   719.3 2192.35
   763.5 2203.93   775.6 2205.63   795.7 2206.01   834.7 2210.57     864 2214.92
   896.2 2216.65   908.3 2217.99   920.3 2217.56   948.5 2218.74   973.6 2221.41
#Mann= 4 ,-1,0
       0     .06       0      50      .1       0   542.8    .045       0
  582.59      .1       0
Bank Sta=542.8,582.59
XS Rating Curve= 0 ,0
Exp/Cntr=0.3,0.1

Type RM Length L Ch R = 1 ,27674   ,553,538.8,512
XS GIS Cut Line= 4
2265075.90589511 691251.897724012265300.88075998691293.445592133
2265677.07258694691341.0610689982265882.56361633691350.504793007
#Sta/Elev= 30
       0 2211.66    65.4 2205.98   134.5 2196.28   211.8 2188.56   240.2 2183.91
     278    2180   312.7 2178.75   328.9 2179.83   362.1 2179.14   449.6 2180.46
     478 2182.68   502.2 2182.92   510.3 2181.74   542.6 2182.12   554.7 2179.13
   566.7 2176.84   586.9 2177.95   590.9 2179.17     599 2183.78   610.5 2193.82
   615.1 2196.81   651.1 2210.02   659.1 2210.43   671.1 2215.29     695 2221.25
   723.2  2227.1   763.2 2232.52   787.2 2237.13   795.3 2239.59   813.7 2242.15
#Mann= 5 ,-1,0
       0      .1       0  438.78     .05       0  538.78      .1       0
   554.7    .045       0   590.9      .1       0
Bank Sta=554.7,590.9
XS Rating Curve= 0 ,0
Exp/Cntr=0.3,0.1

Type RM Length L Ch R = 1 ,27135   ,532.8,558.1,567.6
XS GIS Cut Line= 4
2265117.31033812691748.656361757 2265308.0380294691804.092116961
2265553.56471737691758.1689345922265860.79899367691713.133293797
#Sta/Elev= 30
       0 2256.93    23.8 2257.26    32.1 2251.33    40.5 2241.63    44.6 2239.15
    86.3 2226.48    94.6 2221.52   107.1 2220.34   119.6 2216.85   130.9 2218.13
   136.3 2217.25   169.6 2202.56   180.2  2194.5   202.8 2184.53   235.4 2179.66
   243.5 2176.53   259.8 2175.48  271.412172.207   288.3 2169.64   304.6 2169.17
     329 2169.37  344.522172.208   373.7 2176.87   403.5  2177.3   422.6    2180
   434.8 2179.15   479.3 2183.11   665.3 2210.83   713.8 2219.28   758.9 2229.06
#Mann= 3 ,-1,0
       0      .1       0  271.41    .045       0  344.52      .1       0
Bank Sta=271.41,344.52
XS Rating Curve= 0 ,0
Exp/Cntr=0.3,0.1

Type RM Length L Ch R = 1 ,26577   ,469.1,480.7,489.4
XS GIS Cut Line= 4
2265066.70982909691960.5658249032265266.87427338692182.724421855
2265503.75722458692345.9879529942265761.66171085692459.600872095
#Sta/Elev= 30
       0 2260.79    15.6 2262.46    26.1 2258.56    46.8 2255.56    61.9 2250.09
   117.6 2236.66   193.4 2207.28   230.9 2199.05     270 2184.69   313.2  2172.1
   359.3 2168.98   383.2 2171.74   412.3 2172.99   460.9 2172.94   494.4 2172.24
  529.252168.862   543.5 2165.83   554.8 2165.23  571.912168.861   583.6 2173.59
   604.6 2187.16   619.8 2194.16   727.1 2227.56   753.2 2237.23     797 2248.99
   810.1 2254.46   827.6 2257.97   836.3 2261.33   853.8 2264.03   868.5 2268.53
#Mann= 5 ,-1,0
       0      .1       0  469.03     .05       0  529.25    .045       0
  571.91     .05       0  586.73      .1       0
Bank Sta=529.25,571.91
XS Rating Curve= 0 ,0
Exp/Cntr=0.3,0.1

Type RM Length L Ch R = 1 ,26096   ,426.1,425.3,427.6
XS GIS Cut Line= 4
2264915.55041399692203.4086209782264998.19847926692396.042927284
2265123.82480993692665.5951011682265339.62986108692927.221137065
#Sta/Elev= 30
       0 2232.24    38.4 2226.05    97.7 2210.19   119.4 2201.51   154.1 2189.64
   189.1 2179.31   202.1  2177.3   210.9 2174.59   219.7 2166.87   224.1 2165.06
     255  2164.5   346.9 2167.89   353.4 2167.24   374.2 2169.22   383.5 2167.46
   422.7 2166.06  438.772163.449   449.2 2161.08   466.8  2161.9   470.42163.448
   493.3 2174.58   563.5 2196.08   625.7 2212.66   668.9 2218.93   683.6 2222.81
   722.9 2228.21   737.1 2231.58   805.3 2242.44   827.9 2244.63   846.2 2241.84
#Mann= 4 ,-1,0
       0      .1       0  369.62     .06       0  438.77    .045       0
   470.4      .1       0
Bank Sta=438.77,470.4
XS Rating Curve= 0 ,0
Exp/Cntr=0.3,0.1

Type RM Length L Ch R = 1 ,25671   ,495.8,503.6,508.3
XS GIS Cut Line= 3
     2264541.625      692333.162     2264699.653      692759.837
     2264857.682      693186.513
#Sta/Elev= 30
       0 2196.33    81.1 2192.72    93.9 2187.39   106.7 2186.88   110.9 2185.31
   123.7 2177.23     138 2173.38   160.7 2162.93   166.4 2161.52   183.4 2163.31
   192.2 2162.54   345.5 2163.97   392.4 2166.18   412.9 2163.52     4212160.544
   439.4 2157.69   447.1 2157.65   462.7 2157.95  477.912160.546   490.3 2163.22
   533.2  2164.7   597.2 2163.03   614.3 2165.46   644.1 2177.85   665.4 2183.57
     691 2187.99   708.1 2194.39   734.2 2195.28   793.4 2194.06     910 2205.78
#Mann= 6 ,-1,0
       0      .1       0     220     .06       0     320      .1       0
     421    .045       0  477.91     .06       0     535      .1       0
Bank Sta=421,477.91
XS Rating Curve= 0 ,0
Exp/Cntr=0.3,0.1

Type RM Length L Ch R = 1 ,25167   ,493.6,493,492.8
XS GIS Cut Line= 3
     2264195.038      692438.5582264217.67724815692928.926036977
     2264351.001      693336.036
#Sta/Elev= 30
       0 2174.21    14.6 2175.22    38.7 2174.49    54.7 2175.01   146.8  2171.3
   210.8 2169.98   229.4  2170.3   270.9 2168.91   298.3 2166.86   306.9 2162.44
     315 2160.92     339 2160.69     351 2159.67     359 2160.75   390.2 2160.63
     403 2161.74   415.1 2161.06  431.222157.362   439.1 2155.59   451.1 2154.62
   459.1  2154.9  466.262157.362   475.1 2160.34   483.1 2164.37   495.4 2167.74
   597.7 2173.12   806.8 2177.68   844.1  2179.2     870 2182.64   919.3 2187.63
#Mann= 8 ,-1,0
       0      .1       0     390     .06       0  431.22    .045       0
  466.26     .06       0     490      .1       0  600.89     .05       0
  700.89     .06       0  800.89      .1       0
Bank Sta=431.22,466.26
XS Rating Curve= 0 ,0
Exp/Cntr=0.3,0.1

Type RM Length L Ch R = 1 ,24674   ,519.1,531.9,531.8
XS GIS Cut Line= 3
2263696.65125555692510.1285036982263731.76751109693038.353366478
     2264230.619      693369.533
#Sta/Elev= 30
       0  2161.1   135.3 2157.53   239.2 2157.99   279.7 2154.73   347.8 2156.58
   363.9 2156.06   371.9 2157.94   375.9 2157.69  380.912155.485   387.9 2152.41
   391.9 2151.85   407.9 2151.74     416 2151.91     420 2152.76  426.192155.499
     432 2156.79     452 2156.52   492.1 2158.47   657.4    2160   693.6 2162.97
   741.1 2164.31   789.1 2164.49   808.4 2163.45     866 2163.29     953 2165.45
   981.2 2166.67   995.6 2168.66  1072.4 2170.82  1094.4 2174.13  1128.2 2177.73
#Mann= 12 ,-1,0
       0      .1       0     130     .06       0     220      .1       0
  380.91    .045       0  426.19     .06       0     500     .05       0
     520     .07       0  649.39     .06       0  769.39     .07       0
  869.39     .06       0  999.39     .07       0 1039.39      .1       0
Bank Sta=380.91,426.19
XS Rating Curve= 0 ,0
Exp/Cntr=0.3,0.1

Type RM Length L Ch R = 1 ,24142   ,1096.4,1077,1046.1
XS GIS Cut Line= 3
 2263364.6006454692402.6687700972263272.66071487693089.871299919
2263872.25723007693309.918152011
#Sta/Elev= 30
       0 2157.13    22.7 2156.69    63.1  2154.5   131.7 2155.79   159.9 2155.21
   176.1 2153.91   224.5 2154.51   260.8 2156.16   272.9 2151.97   305.2  2153.9
   347.9 2153.51     511 2154.84   591.7 2154.59   606.5 2153.12   625.5 2150.75
     636 2150.28   644.2  2150.9  650.152153.046   657.5 2155.07   668.4 2156.85
   693.3 2158.91   782.3 2156.62   879.4 2157.66   910.1 2157.12   929.3 2157.89
   995.3 2158.26  1016.6 2160.88  1037.9 2161.97  1080.5  2162.7    1332 2161.05
#Mann= 8 ,-1,0
       0     .06       0     240     .05       0     530      .1       0
   606.5    .045       0  650.15     .05       0  973.33     .06       0
 1083.33     .07       0 1183.33     .05       0
Bank Sta=606.5,650.15
XS Rating Curve= 0 ,0
Exp/Cntr=0.3,0.1

Type RM Length L Ch R = 1 ,23065   ,81.6,86,88.3
XS GIS Cut Line= 6
2262290.95775011692195.5272775712262304.87980004  692365.8574958
 2262370.4216775692552.2157767532262594.29270562692997.422689702
2262969.28581702693144.0933824672263315.81808148693228.781716951
#Sta/Elev= 30
       0 2161.57    69.9 2159.94   109.7 2155.52   237.9  2155.4   246.3 2154.11
     259 2153.95   273.6 2150.72  292.952149.633   301.5 2149.29   314.2 2146.22
     327 2146.06     361 2146.27   379.82149.634   386.8 2151.88     404 2152.87
   533.1 2150.41   604.3 2151.26     671 2150.09   751.4 2151.22   848.1 2149.91
     963 2149.91   992.4 2150.89  1141.1 2152.08  1218.4 2157.12  1282.3 2159.88
  1304.1 2158.93  1525.2 2158.34  1573.2 2159.31  1615.8 2158.88  1627.8 2159.75
#Mann= 12 ,-1,0
       0     .07       0      50     .08       0   250.9     .07       0
  292.95    .045       0   379.8     .07       0  782.26     .06       0
  792.26     .07       0  1035.5     .05       0  1215.5     .08       0
  1245.5     .07       0 1351.07     .08       0 1551.07     .07       0
Bank Sta=292.95,379.8
XS Rating Curve= 0 ,0
Exp/Cntr=0.3,0.1

Type RM Length L Ch R = 1 ,22979   ,773.1,738.7,685.4
XS GIS Cut Line= 6
2262217.10376406692228.5962265482262231.02581399692398.926444777
2262296.56769145692585.2847257312262520.43871957693030.491638679
2262895.43183097693177.1623314442263241.96409543693261.850665928
#Sta/Elev= 30
       0 2160.43    80.9 2158.26     137 2155.78     241 2154.49   270.6 2152.46
  278.532149.443   283.6 2146.49   296.1 2145.81   321.6 2146.09   334.3 2148.95
  340.172149.446   351.3 2151.37   374.2 2152.32   411.7 2151.51   468.6 2151.84
   504.1 2150.52     711 2150.73   786.1 2149.81   926.4 2150.22   947.6 2149.53
   977.3 2150.96  1007.1 2149.78  1115.5  2150.1  1193.3 2153.01    1216 2155.37
    1250 2157.53  1304.8 2158.88  1404.1 2159.29  1514.8 2157.85  1627.8 2158.13
#Mann= 17 ,-1,0
       0     .08       0      10     .07       0     110     .08       0
   210.9     .07       0  278.53    .045       0  340.17     .08       0
  418.45     .07       0  645.96     .06       0  732.26     .07       0
  862.78     .08       0   905.5     .07       0  1115.5     .05       0
  1125.5     .08       0 1321.07     .07       0 1421.07     .08       0
 1461.07     .06       0 1531.07     .07       0
Bank Sta=278.53,340.17
XS Rating Curve= 0 ,0
Exp/Cntr=0.3,0.1

Type RM Length L Ch R = 1 ,22240   ,321.6,321,319.8
XS GIS Cut Line= 4
2261880.03310928693186.6221432332262197.38510147693106.399463356
2262816.87555738693184.3181214482263230.43524779693288.678525024
#Sta/Elev= 30
       0 2182.32    49.7 2181.74    74.4 2180.43   107.4 2176.75   111.5 2174.78
   123.9 2165.08   139.6  2154.8   152.8 2151.56  245.242148.458   251.8 2144.97
   268.1 2144.22   293.1 2144.54  299.072148.457   309.6 2150.04   350.4 2149.99
   362.4 2148.56   382.6 2148.75     415 2146.87   475.3 2149.97   559.9 2149.39
   624.4 2151.57   726.2  2149.4   812.2  2149.2   842.1 2151.67   918.7 2151.13
   975.7 2156.59  1098.5 2158.97    1182 2158.52  1268.1 2156.08  1378.2 2156.78
#Mann= 10 ,-1,0
       0     .05       0      90      .1       0  245.24    .045       0
  299.07      .1       0  487.33     .05       0  587.33     .08       0
 1081.71     .07       0 1111.71      .1       0 1191.71     .06       0
 1291.71     .07       0
Bank Sta=245.24,299.07
XS Rating Curve= 0 ,0
Exp/Cntr=0.3,0.1

Type RM Length L Ch R = 1 ,21919   ,1156,1153,1116.8
XS GIS Cut Line= 3
2262075.12006544693472.737774901 2262816.0417561693253.000801528
2263205.98731935 693303.10718671
#Sta/Elev= 30
       0 2199.38     9.4  2198.9    26.1 2189.99    42.8 2182.93    67.9 2167.79
    84.5  2154.6    88.7  2152.3   109.6 2151.87   113.7 2150.97  120.122147.407
   129.2 2144.27   142.1 2144.04   167.8 2147.36   205.5 2148.71   277.2 2146.56
   343.2 2149.25     422 2149.84   502.5 2149.09   595.3 2149.92   647.8 2148.38
   672.4 2150.41   706.2 2150.38   731.2 2154.28   756.3 2153.41     777 2155.14
   833.8 2157.05   986.7 2156.77  1079.5 2154.98    1148    2155    1166 2156.11
#Mann= 10 ,-1,0
       0     .05       0      90      .1       0  120.12    .045       0
   167.8      .1       0     400     .05       0     540     .06       0
     700     .07       0  902.82      .1       0 1002.82     .06       0
 1102.82     .07       0
Bank Sta=120.12,167.8
XS Rating Curve= 0 ,0
Exp/Cntr(USF)=0,0
Exp/Cntr=0.3,0.1

Type RM Length L Ch R = 1 ,20767   ,74.6,59.2,50.6
XS GIS Cut Line= 6
2262452.08922027694154.9094755712262932.80778848693860.424751905
2262861.77078698693715.901197116 2262762.2745255693488.816479535
2262682.08270679693349.4882426152262908.89305643693301.102034693
#Sta/Elev= 30
       0 2235.55    28.2 2223.58      75 2200.06    94.5 2192.53     119 2185.34
   131.1 2185.04   149.8 2187.75   154.5 2186.73   163.8 2182.84   187.7  2166.9
   219.7 2155.91   240.1 2151.51   262.1 2149.82     310  2148.4   534.2  2149.6
   665.3 2147.56   854.6 2147.54  880.052146.352   908.4 2142.88   928.8 2142.69
     955 2142.99  968.612146.353   977.1 2148.59  1044.7 2148.54  1115.4 2150.03
  1168.5 2148.47  1250.4 2152.51    1279 2152.45  1334.6 2155.21  1365.6 2155.64
#Mann= 11 ,-1,0
       0     .05       0     100      .1       0     350     .06       0
  622.55     .07       0  734.98     .06       0  774.98     .07       0
  844.98     .06       0  880.05    .045       0  968.61     .07       0
  1012.9     .06       0 1203.67     .07       0
Bank Sta=880.05,968.61
XS Rating Curve= 0 ,0
Exp/Cntr(USF)=0,0
Exp/Cntr=0.3,0.1

Type RM Length L Ch R = 1 ,20707   ,759.2,794.5,817.7
XS GIS Cut Line= 6
2262505.83212589694155.201431059 2262986.5506941693860.716707393
 2262915.5136926693716.1931526042262816.01743112693489.108435023
2262735.82561241693349.7801981032262962.63596205693301.393990181
#Sta/Elev= 30
       0 2207.14    40.2 2191.81    61.4  2186.7    72.9    2186    96.5 2188.95
   104.2 2188.59   122.6 2180.86   138.4 2169.49   148.8 2164.53   173.6    2157
   195.4 2151.92   212.8 2151.02   222.6 2149.12   311.9 2148.15   483.7 2149.35
   634.7 2146.87   679.3 2146.85   692.7 2148.28   723.9  2147.1  957.912146.115
   972.5 2144.85   981.5 2142.71   991.2  2142.5  1004.9 2142.72  1013.22146.118
  1022.7 2149.64  1133.7 2149.24  1256.7 2152.52  1289.4 2155.18  1365.6  2154.6
#Mann= 16 ,-1,0
       0     .05       0     100      .1       0     280     .05       0
     290     .06       0  622.55     .07       0  734.98     .06       0
  844.98     .05       0  904.98     .06       0  944.98     .07       0
  957.91    .045       0  1013.2     .07       0 1119.68     .06       0
 1143.67     .07       0 1253.67     .05       0 1283.67     .07       0
 1353.67      .1       0
Bank Sta=957.91,1013.2
XS Rating Curve= 0 ,0
Exp/Cntr(USF)=0,0
Exp/Cntr=0.3,0.1

Type RM Length L Ch R = 1 ,19913   ,1407.9,1454.6,1492.3
XS GIS Cut Line= 4
2262724.57953187694340.2525531162263122.13711475694219.607469613
2263596.43605273693555.2475294952263589.34561756693424.574191643
#Sta/Elev= 30
       0 2167.42    16.3 2163.29    37.2 2161.14    53.9 2152.11    62.3 2151.13
     108 2151.66   129.2  2154.6   162.6 2155.76   304.7 2151.01   570.4  2149.6
   607.9 2148.43   654.4 2145.28   719.8 2145.51   804.5 2147.39   841.1  2146.8
   868.9 2143.65   894.7  2144.3   906.1 2141.15   923.4 2140.73   937.7 2141.26
   944.3 2144.34   949.2 2145.28   993.5 2143.43  1058.1 2145.44  1081.9 2143.67
  1149.9 2143.83  1162.5 2144.42  1175.3  2148.3  1210.1 2153.82  1362.6 2159.12
#Mann= 10 ,-1,0
       0      .1       0     130     .05       0     340     .06       0
  435.46     .05       0  555.46     .06       0  615.46     .03       0
  675.46     .05       0   894.7    .045       0   944.3      .1       0
 1271.75     .07       0
Bank Sta=894.7,944.3
XS Rating Curve= 0 ,0
Exp/Cntr=0.3,0.1

Type RM Length L Ch R = 1 ,18458   ,695.7,663.7,622.5
XS GIS Cut Line= 6
2262968.71400479694383.4746559782263088.10380173 694464.27356536
2263276.48363389694543.0560308982263308.65143857694582.369824836
2263609.50438478694689.8888958942263897.38565733694516.858710929
#Sta/Elev= 30
       0  2159.8    88.7 2155.38   139.1 2153.91   156.9 2151.75   183.3 2146.88
   204.9 2144.73   239.6 2144.07   248.9 2142.68   265.6  2141.7   328.3 2143.85
   343.7 2142.86     3492141.037   356.3 2139.56   372.4  2139.5   382.1 2139.64
  389.142141.051   395.1 2142.95   407.2 2143.35   429.1 2146.05     473 2146.26
   500.6 2147.58   525.9 2147.81   653.5 2147.35   704.5 2149.29   754.4 2152.46
   836.5 2154.97   889.8 2156.14   927.1  2155.3  1011.1 2158.75  1054.5 2161.35
#Mann= 6 ,-1,0
       0     .05       0  314.16      .1       0     349    .045       0
  389.14      .1       0  748.64     .06       0  978.64      .1       0
Bank Sta=349,389.14
XS Rating Curve= 0 ,0
Exp/Cntr=0.3,0.1

Type RM Length L Ch R = 1 ,17795   ,163.3,162.3,157.4
XS GIS Cut Line= 5
2263160.64537566 695133.832962562263342.11926847694955.720199589
2263476.40465371694821.0921159312263703.17635851 694750.90803993
2263819.22398521694666.486740581
#Sta/Elev= 30
       0 2220.51    22.8 2217.28    63.7 2195.27    94.6 2190.71   152.9 2179.34
   178.7 2173.14   189.4 2168.33   200.8 2167.05   235.1 2153.76   243.4 2147.12
   246.2 2145.96   262.9 2145.59   271.7 2147.74   274.8 2147.21   285.8 2141.94
   302.8 2140.92   311.3 2141.57   319.5  2140.1   336.5 2138.91  376.682140.092
   390.5  2141.9   404.8 2140.79   427.1 2145.45   435.7 2144.53   498.6 2145.03
     641  2152.3   697.9 2154.03   727.6 2156.34   773.1 2157.54   825.3 2157.29
#Mann= 6 ,-1,0
       0      .1       0   319.5    .045       0  376.68      .1       0
  614.43     .06       0  721.81      .1       0  781.81     .06       0
Bank Sta=319.5,376.68
XS Rating Curve= 0 ,0
Exp/Cntr=0.3,0.1

Type RM Length L Ch R = 1 ,17632   ,490.5,464.1,427.8
XS GIS Cut Line= 4
2263366.69243164695224.9444114922263484.72012633 695046.30089781
2263581.27863704694929.6198907772263850.76004312694677.201599951
#Sta/Elev= 30
       0 2241.13     4.5 2239.63    17.2 2231.38    33.3 2217.07    57.2 2199.88
    70.2 2193.32   162.6 2162.45   172.3 2156.97   191.4 2154.94   205.9 2150.25
   214.5  2144.8   236.3 2143.71   246.7 2141.28   263.4 2141.28  275.312139.808
   285.5 2138.31   307.4 2138.03   324.6 2138.41  329.062139.809     345 2143.45
   372.1 2147.04   396.9  2146.1   418.9 2149.09   462.7 2148.53   537.7 2154.95
     549 2154.12     571 2155.78   645.3 2157.82   692.9 2157.16   734.8 2158.36
#Mann= 5 ,-1,0
       0      .1       0  275.31    .045       0  329.06      .1       0
  435.57     .06       0  575.57      .1       0
Bank Sta=275.31,329.06
XS Rating Curve= 0 ,0
Exp/Cntr=0.3,0.1

Type RM Length L Ch R = 1 ,17168   ,493.1,542,575
XS GIS Cut Line= 4
2263995.59099849695349.1274992472264001.56045708695070.815004157
2263924.64194747694866.6697218522263894.02530409694737.712569525
#Sta/Elev= 30
       0 2219.17      12 2216.37    40.2 2199.94    72.9 2187.13     124 2175.15
     132 2175.19     160 2171.09     172    2169     184 2163.59     200 2163.07
     220 2165.54     240 2164.91     252 2163.69     260  2161.1   273.3 2157.83
   277.4 2153.61   284.4 2142.04   288.7 2136.97     290 2136.51   305.6  2135.7
   318.6 2138.04   327.1 2138.09   347.4 2131.11   365.6 2128.96   407.1 2129.24
  420.742131.111   459.7 2137.36   468.2 2137.18   514.5  2143.7   629.1 2156.23
#Mann= 5 ,-1,0
       0      .1       0     160     .06       0     260      .1       0
   347.4    .045       0  420.74      .1       0
Bank Sta=347.4,420.74
XS Rating Curve= 0 ,0
Exp/Cntr=0.3,0.1

Type RM Length L Ch R = 1 ,16626   ,568.8,575.7,593.2
XS GIS Cut Line= 4
2264214.07638332695354.4098567762264362.08217313695054.366040129
2264494.28417657694933.3894256142264561.82899083694798.841094208
#Sta/Elev= 30
       0 2182.08    23.7 2177.33    44.3 2176.77   112.9 2169.89   170.9  2167.3
   175.3 2166.16   184.2 2153.06   188.7 2148.53   193.2 2146.39   202.1 2145.03
   260.1 2140.04   277.9 2139.85   303.1 2136.74   319.1  2136.6   331.4 2134.05
   353.9 2135.03   375.4 2130.31  396.412127.425   418.7 2124.08   433.1 2123.98
     453  2125.1  462.422127.426   472.9 2130.68     514 2136.28   549.8 2143.52
     569 2149.05   594.6 2159.67   625.9 2167.92   643.8  2174.7   664.3 2176.05
#Mann= 4 ,-1,0
       0     .06       0      80      .1       0  396.41    .045       0
  462.42      .1       0
Bank Sta=396.41,462.42
XS Rating Curve= 0 ,0
Exp/Cntr=0.3,0.1

Type RM Length L Ch R = 1 ,16051   ,394.1,392.7,400.3
XS GIS Cut Line= 4
2264350.81244822695538.3177063512264661.65703251 695461.34143423
2264887.37866511695392.3851385662265148.21074187695277.555763401
#Sta/Elev= 30
       0 2180.91     8.7 2180.52    59.1 2173.05    75.6  2172.8    91.2 2170.22
   116.8 2168.49   120.9 2166.19   129.1 2149.22   133.3 2146.19   167.2 2141.79
   252.8 2134.47   269.3 2133.75   277.5 2134.63   289.4 2132.18   339.6  2129.5
   368.9 2128.84   414.9 2129.87   452.5 2126.38  459.052124.328   469.3 2121.52
     489 2120.73   506.9 2121.63  515.382124.329   544.5 2132.95   565.9 2141.02
   616.9 2157.21   653.3 2164.73   692.6 2175.27   727.6 2180.69   841.2 2192.16
#Mann= 4 ,-1,0
       0     .06       0      70      .1       0  459.05    .045       0
  515.38      .1       0
Bank Sta=459.05,515.38
XS Rating Curve= 0 ,0
Exp/Cntr=0.3,0.1

Type RM Length L Ch R = 1 ,15658   ,617.2,576.2,550.2
XS GIS Cut Line= 4
2264394.89016872695785.1343990712264658.49956562695821.724191018
2264904.72451704695793.4183390412265043.92509093695633.705979189
#Sta/Elev= 30
       0 2184.36    49.8 2174.02    65.9 2168.75    90.1  2167.5   122.4 2160.93
   126.5 2159.08   134.6 2150.71   138.6 2148.24     179 2139.23   266.1 2129.81
     288 2128.51     300  2130.7   312.1 2130.44   324.2 2126.88   332.2 2125.72
   368.5 2124.41  379.032123.007   399.4 2120.21   412.6 2119.53     449 2119.81
  461.322123.008   481.1 2126.75   530.2 2142.16   556.7 2146.28   570.5 2150.27
   601.7 2161.64   634.9 2168.47     664 2178.87   701.9 2182.73   725.8 2183.62
#Mann= 5 ,-1,0
       0      .1       0      30     .06       0     130      .1       0
  379.03    .045       0  461.32      .1       0
Bank Sta=379.03,461.32
XS Rating Curve= 0 ,0
Exp/Cntr=0.3,0.1

Type RM Length L Ch R = 1 ,15082   ,469.4,476.6,482.5
XS GIS Cut Line= 4
2264854.00013174696382.7500947662265091.46637304696138.074059248
2265262.80935326695932.3271513282265347.33481895695792.425896749
#Sta/Elev= 30
       0 2172.75    35.6 2171.18    47.9 2165.91    62.1 2164.31   138.4 2148.46
   152.5 2146.98   197.3 2138.99   230.7 2136.73   243.1 2134.75     253 2129.74
   255.8 2129.14   269.7    2129   286.5 2130.43     294  2129.6   378.6 2126.01
   420.2 2124.77   475.6 2124.25   495.5 2122.91  516.142120.246   542.1 2117.56
   571.2 2117.91  578.612120.248     592  2128.6   617.8 2141.08   663.8  2156.6
     681 2161.67   719.6  2169.3   743.2 2171.77   752.6 2169.21   772.2 2167.56
#Mann= 3 ,-1,0
       0      .1       0  516.14    .045       0  578.61      .1       0
Bank Sta=516.14,578.61
XS Rating Curve= 0 ,0
Exp/Cntr=0.3,0.1

Type RM Length L Ch R = 1 ,14605   ,429.7,440.4,453.4
XS GIS Cut Line= 4
2265064.61307104 696565.91687944 2265331.3487805696464.772702798
2265496.09912154696342.2480161432265627.89210361696138.460313392
#Sta/Elev= 30
       0 2181.91    80.8 2178.95   102.6 2176.45   119.3  2176.6   136.4 2173.76
   158.4 2167.52   162.1 2164.92   170.6 2154.08   177.1 2151.04   247.7 2137.82
   282.5 2124.06   316.2 2123.86  331.892115.977   361.1 2113.06   391.8 2113.78
  401.762115.977   415.9 2120.83   470.7 2123.26   501.4 2126.15   511.7 2128.27
   542.3 2128.34   552.2 2130.06   577.6 2130.41   596.7 2131.86   608.6 2134.42
   620.5 2132.93   639.5 2134.24   673.7 2143.02   720.5 2158.23   733.3 2160.15
#Mann= 4 ,-1,0
       0      .1       0  331.89    .045       0  401.76      .1       0
  580.59     .12       0
Bank Sta=331.89,401.76
XS Rating Curve= 0 ,0
Exp/Cntr=0.3,0.1

Type RM Length L Ch R = 1 ,14165   ,507.1,495.8,480.5
XS GIS Cut Line= 4
2265221.35667488696847.9917449982265528.59544122696804.222152394
2265739.22677569696758.299133567 2265927.6196957696679.367061629
#Sta/Elev= 30
       0 2175.95    63.5  2165.5    67.5  2164.3    79.6 2154.76   111.9 2147.65
   176.6 2140.03   212.9 2133.45   305.6 2123.66   326.3 2123.66   338.6  2120.1
   354.9 2120.13   375.4 2115.65   402.32113.146   416.4 2110.59   430.2 2110.41
   453.2 2111.41  457.722113.146   539.2 2132.64   557.3 2138.69     566 2143.28
   574.7 2143.83   591.7 2154.23   600.7 2157.48   622.2 2169.56   635.4 2174.83
   687.4 2182.15   696.1 2184.38   700.4 2187.68   717.8 2205.68   730.2 2211.25
#Mann= 4 ,-1,0
       0      .1       0   402.3    .045       0  457.72      .1       0
  695.92     .12       0
Bank Sta=402.3,457.72
XS Rating Curve= 0 ,0
Exp/Cntr=0.3,0.1

Type RM Length L Ch R = 1 ,13669   ,487.3,504.8,513.5
XS GIS Cut Line= 4
2265482.98205916697451.2661668012265711.18278674697303.535721765
 2265865.8037189697170.4863099422266042.75713722696989.487314711
#Sta/Elev= 30
       0 2165.83    34.8 2166.79      92 2171.35   125.3 2172.76   143.7 2172.17
   151.1 2168.78   158.4 2154.85   161.5 2151.09   177.7 2144.32   234.9 2127.65
     254 2124.59   287.7 2114.68   311.1 2116.06  324.062109.601   330.9 2107.37
   341.8 2106.97   362.9 2107.16   377.7  2109.6   389.2 2113.56   418.9 2115.92
   438.7 2120.66   488.8 2121.22   522.4 2129.29   544.8 2136.68   570.8 2141.23
   622.7 2160.28   693.4 2180.12   707.5 2185.33   723.8 2187.44     729 2190.03
#Mann= 5 ,-1,0
       0      .1       0  324.06    .045       0   377.7      .1       0
  635.83     .12       0  665.83      .1       0
#XS Ineff= 2 , 0
          302.09 2136.09
Permanent Ineff=
       F       F
Bank Sta=324.06,377.7
XS Rating Curve= 0 ,0
Exp/Cntr=0.3,0.1

Type RM Length L Ch R = 1 ,13164   ,518.1,493.1,468.1
XS GIS Cut Line= 4
2265784.51793808697584.0116415072265994.49934611697577.247692303
2266158.91761666697567.6948948982266430.29208198697541.361349322
#Sta/Elev= 30
       0 2160.94    39.7 2157.31    67.7 2152.75    99.7 2143.94   135.7  2131.9
   166.3 2124.34   184.6 2116.74   199.8 2116.81   211.8 2115.31   227.8 2111.76
   235.8 2108.92   247.8 2110.35   267.9    2111   283.7 2108.72  295.822105.605
   307.9 2103.24     320 2102.71     332 2102.95  338.872105.607     360 2116.22
   388.1 2123.07   404.2 2128.88   444.4  2134.6   452.4 2136.91   496.6 2145.33
   524.8 2149.23   548.9  2154.8     589 2162.19   609.1 2167.27   647.4 2172.28
#Mann= 3 ,-1,0
       0      .1       0  295.82    .045       0  338.87      .1       0
#XS Ineff= 2 , 0
          261.11 2132.96
Permanent Ineff=
       F       F
Bank Sta=295.82,338.87
XS Rating Curve= 0 ,0
Exp/Cntr=0.3,0.1

Type RM Length L Ch R = 1 ,12671   ,497.9,494.8,491.9
XS GIS Cut Line= 3
     2265889.174      698359.3712266211.90375578697993.875051023
2266482.89601684697748.720839936
#Sta/Elev= 30
       0  2156.2    18.9 2154.78    56.3 2154.87      71 2153.39    77.4 2150.17
     115 2140.57   317.8 2119.65   332.4 2112.71   343.7 2112.22   355.1 2113.97
   376.5 2108.42   386.3 2107.56  409.99 2100.17   420.3 2098.34   463.8 2097.73
  476.412100.171   496.8 2110.27   506.5 2118.33   513.8 2120.93   563.5 2129.77
   587.4 2131.26   633.6 2137.12   643.6 2141.45   660.6 2144.96   692.9 2157.01
   715.2 2166.78   727.1 2174.52   736.1 2177.53   794.1 2181.09     853 2188.03
#Mann= 5 ,-1,0
       0     .06       0      30      .1       0  409.99    .045       0
  476.41      .1       0  727.59     .08       0
Bank Sta=409.99,476.41
XS Rating Curve= 0 ,0
Exp/Cntr=0.3,0.1

Type RM Length L Ch R = 1 ,12176   ,505.2,509.8,513.9
XS GIS Cut Line= 4
2266328.82243742698605.961227212 2266545.3414232698333.296132917
2266664.91594898698186.0145765342266760.43070802 697969.50260477
#Sta/Elev= 30
       0 2174.63    31.1  2170.4    42.8  2164.3    57.2 2161.36   123.6 2153.48
   133.8 2150.16     151 2149.68   205.3 2139.37   241.1 2120.36   266.6 2117.94
     327 2107.13   338.1 2101.91   350.3 2101.64   368.9 2092.36   427.1 2094.68
   438.4 2093.88  451.312089.769   485.9 2087.62   497.7 2090.59  507.092089.769
   535.1  2099.5   573.8 2106.01   613.1 2118.09   643.7 2130.81   661.2 2149.34
   664.9 2150.57   710.9 2157.81   735.1 2158.84   761.8 2169.64   774.5 2172.05
#Mann= 4 ,-1,0
       0      .1       0  451.31    .045       0  507.09      .1       0
  697.89     .08       0
Bank Sta=451.31,507.09
XS Rating Curve= 0 ,0
Exp/Cntr=0.3,0.1

Type RM Length L Ch R = 1 ,11666   ,502.2,490.1,473.7
XS GIS Cut Line= 3
 2266720.8598332698824.9908567762267068.19136765698516.088727862
2267164.09340016698271.583839936
#Sta/Elev= 30
       0 2193.44      39 2195.84    59.9 2199.88   138.3 2201.13   143.9 2195.63
   149.5 2173.41   156.2  2158.6   175.7 2149.06   211.9 2136.75   216.4 2132.32
   228.4 2113.42     240 2106.13   279.9 2092.94   294.6 2091.62  322.342079.716
     347 2077.43  374.162079.713     438 2085.97   451.1 2089.66   473.2 2089.42
   502.3 2094.72   510.9 2100.82     538 2099.62   575.4 2105.57   593.6 2130.72
   605.4 2139.66   626.9 2147.08   691.4 2154.95   710.9 2167.67   727.5 2174.53
#Mann= 3 ,-1,0
       0      .1       0  322.34    .045       0  374.16      .1       0
Bank Sta=322.34,374.16
XS Rating Curve= 0 ,0
Exp/Cntr=0.3,0.1
